HEC-RAS study C100-00-00.prj: C100-00-00

--- C100-00-00.g01 (geometry) --- (continued)

Type RM Length L Ch R = 3 ,106678  ,,,
BEGIN DESCRIPTION:
BLUE RIDGE ROAD
Structure ID: C00-48
END DESCRIPTION:
Bridge Culvert--1,0,-1,-1, 0
Deck Dist Width WeirC Skew NumUp NumDn MinLoCord MaxHiCord MaxSubmerge Is_Ogee
10,28,2.6,0, 48, 48, , , 0.95, 0, 1,1,,
    4227    4252    4267    4317    4332    4347  4375.9  4410.9  4430.9  4490.9
  4620.9  4645.9  4660.9  4710.9  4720.9  4735.7  4761.4    4782  4833.3  4889.8
  4897.6  4924.9  4951.5  4952.7  4953.2  4972.9  5039.1  5042.5    5096  5155.9
  5221.1  5277.7  5310.9  5350.9  5361.4  5441.5  5501.4  5561.4  5636.4  5683.4
  5728.4  5743.4  5788.4  5998.4  6058.4  6333.4  6353.4    6455
    64.4      64    64.4    63.7    63.9    63.5    63.8    63.1    63.5    63.7
    61.7    60.4      60   60.25   60.32   60.42    60.6   61.22   61.87    62.1
    62.2   62.53    62.7    62.7    62.7   62.67   62.59   62.59   62.45   62.47
   62.54   62.43   62.26   62.05      62   62.06    62.1    62.3    62.2   62.01
    61.5    62.1    61.8    62.8    62.4    62.7    63.2    63.5
    64.4      64    64.4    63.7    63.9    63.5    63.8    63.1    63.5    63.7
    61.7    60.4      60    60.1    59.8   59.65   59.02   58.52   59.72   60.78
   61.04   61.65    60.8    60.8   60.98   60.77   60.69   61.31   59.74   60.57
   60.64   60.44    61.5    60.6   60.69    61.4   61.52   61.65    61.8    61.9
    61.5    62.1    61.8    62.8    62.4    62.7    63.2    63.5
    4227    4252    4267    4317    4332    4347  4375.9  4410.9  4430.9  4490.9
  4620.9  4645.9  4660.9  4710.9  4720.9  4735.7  4761.4    4782  4833.3  4889.8
  4897.6  4924.9  4951.5  4952.7  4953.2  4972.9  5039.1  5042.5    5096  5155.9
  5221.1  5277.7  5310.9  5350.9  5361.4  5441.5  5501.4  5561.4  5636.4  5683.4
  5728.4  5743.4  5788.4  5998.4  6058.4  6333.4  6353.4    6455
   64.48   64.08   64.48   63.78   63.98   63.58   63.88   63.18   63.58   63.78
   61.78   60.48   60.08   60.25   60.32   60.42    60.6   61.22   61.87    62.1
    62.2   62.53    62.7    62.7    62.7   62.67   62.59   62.59   62.45   62.47
   62.54   62.43   62.26   62.05      62   62.06    62.1    62.3    62.2   62.01
   61.58   62.18   61.88   62.88   62.48   62.78   63.28   63.58
   64.48   64.08   64.48   63.78   63.98   63.58   63.88   63.18   63.58   63.78
   61.78   60.48   60.08   60.18   59.88   59.73    59.1    58.6    59.8   60.86
   61.12   61.73   60.88   60.88   61.06   60.85   60.77   61.39   59.82   60.65
   60.72   60.52   61.58   60.68   60.77   61.48    61.6   61.73   61.88   61.98
   61.58   62.18   61.88   62.88   62.48   62.78   63.28   63.58
Pier Skew, UpSta & Num, DnSta & Num=  ,4982.1, 2 ,4982.1, 2 , 0 , 0 , 0 ,,
     1.4     1.4
   50.62   61.76
     1.4     1.4
    50.7   61.84
Pier Skew, UpSta & Num, DnSta & Num=  ,5012.3, 2 ,5012.3, 2 , 0 , 0 , 0 ,,
     1.4     1.4
   49.18   61.73
     1.4     1.4
   49.26   61.81
Abutment Skew #Up #Dn= , 2 , 2
  4951.5  4986.8
    60.8   49.78
  4951.5  4986.8
   60.88   49.86
Abutment Skew #Up #Dn= , 2 , 2
  5021.9 5042.79
   53.82    61.3
  5021.9 5042.79
    53.9   61.38
BR Coef= 1 , 1 , 0 ,1.25, 0 ,,,0.8,0,2,0,
WSPro=,,,, 1 ,,,, 0 ,,,, 0 ,,,,-1 ,-1 ,-1 , 0 , 0 , 0 , 0 , 0
BR U #Sta/Elev= 91
    4227    64.4    4252      64    4267    64.4    4317    63.7    4332    63.9
    4347    63.5  4375.9    63.8  4410.9    63.1  4430.9    63.5  4490.9    63.7
  4620.9    61.7  4645.9    60.4  4660.9      60  4661.4      60  4710.9    60.1
  4720.9    59.8  4735.7   59.65  4761.4   59.02  4781.8   58.52    4782   58.52
  4833.3   59.72  4833.4   59.72  4888.8   60.75  4889.8   60.78  4897.6   61.04
  4924.9   61.65    4925   61.65  4951.5    60.8 4951.61   60.79  4951.7   60.79
  4951.9   60.79  4952.7   60.76  4953.2   60.98    4971   54.13  4972.9   53.21
  4982.1   51.95  4986.7   49.78  4986.8   49.78  4990.8   49.82  4995.6   49.76
  4996.1   49.24  4996.2   48.73  4996.9   48.41  4998.3    48.2  5000.8   48.43
  5002.2   48.87  5003.2    48.6  5003.7   49.44    5004   49.65  5008.4   50.58
  5009.5    50.5  5012.3   50.07  5018.4   52.77  5021.8   53.81  5021.9   53.82
  5024.3   54.07  5039.1   60.44    5042    61.2  5042.4   61.31  5042.5   61.31
 5042.59    61.3  5042.7    61.3  5095.8   59.75    5096   59.74  5097.6   59.75
  5155.9   60.57  5156.6   60.57  5221.1   60.64    5223   60.63  5277.7   60.44
  5278.6   60.47  5291.5    60.9  5310.9    61.5  5350.9    60.6  5361.4   60.69
  5441.5    61.4  5501.4   61.52  5561.4   61.65  5636.4    61.8  5683.4    61.9
  5686.4   61.87  5686.5   61.87  5728.4    61.5  5743.4    62.1  5788.4    61.8
  5998.4    62.8  6058.4    62.4  6333.4    62.7  6347.6   63.06  6353.4    63.2
    6455    63.5
BR U #Mann= 4
    4227     .06  4953.2    .035  5042.4     .08  6347.6      .2
BR U Banks=4953.2,5042.4
BR D #Sta/Elev= 91
    4227   64.48    4252   64.08    4267   64.48    4317   63.78    4332   63.98
    4347   63.58  4375.9   63.88  4410.9   63.18  4430.9   63.58  4490.9   63.78
  4620.9   61.78  4645.9   60.48  4660.9   60.08  4661.4   60.08  4710.9   60.18
  4720.9   59.88  4735.7   59.73  4761.4    59.1  4781.8    58.6    4782    58.6
  4833.3    59.8  4833.4    59.8  4888.8   60.83  4889.8   60.86  4897.6   61.12
  4924.9   61.73    4925   61.73  4951.5   60.88 4951.61   60.87  4951.7   60.87
  4951.9   60.87  4952.7   60.84  4953.2   61.06    4971   54.21  4972.9   53.29
  4982.1   52.03  4986.7   49.86  4986.8   49.86  4990.8    49.9  4995.6   49.84
  4996.1   49.32  4996.2   48.81  4996.9   48.49  4998.3   48.28  5000.8   48.51
  5002.2   48.95  5003.2   48.68  5003.7   49.52    5004   49.73  5008.4   50.66
  5009.5   50.58  5012.3   50.15  5018.4   52.85  5021.8   53.89  5021.9    53.9
  5024.3   54.15  5039.1   60.52    5042   61.28  5042.4   61.39  5042.5   61.39
 5042.59   61.38  5042.7   61.38  5095.8   59.83    5096   59.82  5097.6   59.83
  5155.9   60.65  5156.6   60.65  5221.1   60.72    5223   60.71  5277.7   60.52
  5278.6   60.55  5291.5   60.98  5310.9   61.58  5350.9   60.68  5361.4   60.77
  5441.5   61.48  5501.4    61.6  5561.4   61.73  5636.4   61.88  5683.4   61.98
  5686.4   61.95  5686.5   61.95  5728.4   61.58  5743.4   62.18  5788.4   61.88
  5998.4   62.88  6058.4   62.48  6333.4   62.78  6347.6   63.14  6353.4   63.28
    6455   63.58
BR D #Mann= 4
    4227     .06  4953.2    .035  5042.4     .08  6347.6      .2
BR D Banks=4953.2,5042.4
BC Design=,, 0 ,, 0 ,,,,,,
BC HTab HWMax=64.45
BC Use User HTab Curves=0
BC User HTab FreeFlow(D)= 0

Type RM Length L Ch R = 1 ,106654  ,712.21,708.99,705.82
BEGIN DESCRIPTION:
Downstream Section of Bridge/Culvert/Weir
END DESCRIPTION:
XS GIS Cut Line= 4
       3082511.5     13792632.33      3082514.85     13792117.29
      3082564.23     13791299.79       3082312.8     13790441.92
#Sta/Elev= 30
    4227   64.56  4410.9   63.26  4490.9   63.86  4620.9   61.86  4660.9   60.16
  4710.9   60.26  4781.8   58.68  4924.9   61.81  4953.2   61.14  4972.9   53.37
  4982.1   52.11  4986.7   49.94  4995.6   49.92  4996.2   48.89  4998.3   48.36
  5003.2   48.76    5004   49.81  5008.4   50.74  5012.3   50.23  5042.4   61.47
    5096    59.9  5155.9   60.73  5277.7    60.6  5310.9   61.66  5350.9   60.76
  5441.5   61.56  5728.4   61.66  5998.4   62.96  6347.6   63.22    6455   63.66
#Mann= 4 , 1 , 0
    4227     .06       0  4953.2    .035       0  5042.4     .08       0
  6347.6      .2       0
#XS Ineff= 2 , 0
       0    4954      60    5053       0   61.99
Permanent Ineff=
       F       F
Bank Sta=4953.2,5042.4
XS Rating Curve= 0 ,0
Exp/Cntr=0.5,0.3

Type RM Length L Ch R = 1 ,105945  ,899.08,903.42,905.93
BEGIN DESCRIPTION:
Cross Section 108043.1-Interpolated
END DESCRIPTION:
XS GIS Cut Line= 5
        3083130.     13794050.26      3083237.99     13792106.49
      3083237.99     13791904.02      3083237.99     13790338.21
      3082671.06     13788920.88
#Sta/Elev= 30
  2828.3      66  3023.3    61.8    3367   60.49  3508.1   59.82  3578.3    60.9
  3683.3    58.8  3728.3    61.8  3803.3    62.7  3983.3    59.2  4028.3    61.7
  4223.3    61.8  4508.3      59  4613.3    62.2  4658.3    59.3  4739.8   59.73
  4763.3    57.8  4795.1    50.9  4870.1    63.3  4930.1    62.1  4975.1    49.8
  5000.5   47.61  5029.1   55.71  5040.7    61.5  5062.5      63  5762.5    61.2
  5812.5    64.7  6002.5    64.7  6047.5    61.8  6325.6   61.93  8069.9    62.7
#Mann= 7 , 1 , 0
  2828.3      .2       0    3367     .06       0  3508.1      .1       0
  4739.8     .06       0  4930.1    .035       0  5040.7     .06       0
  6325.6      .2       0
Bank Sta=4930.1,5040.7
XS Rating Curve= 0 ,0
Exp/Cntr=0.3,0.1

Type RM Length L Ch R = 1 ,105041.6,350.36,354.39,358.32
BEGIN DESCRIPTION:
Cross Section  107139.5
END DESCRIPTION:
XS GIS Cut Line= 6
      3084041.23     13795025.71      3084201.25     13793125.53
      3084131.24     13792075.43      3084151.24      13791745.4
      3084051.23     13790815.31      3083181.15     13788950.14
#Sta/Elev= 30
  1873.6    64.9  2158.6    63.9  2308.6    61.1  2678.6    62.5  2748.6    61.4
  3303.6    60.4  3389.3   61.96  3468.6    58.6  3483.6    58.9  3513.6    61.3
  4731.6   62.07    4869    63.1  4946.5   62.18  4978.2   48.62  4996.2   47.25
  4997.1   46.29  5000.5   46.12  5002.8   46.23  5004.8   48.64  5029.1   54.22
  5040.7   60.01  5080.8   62.29    5094    59.8  5164.7    61.2  6100.1    64.6
  6295.1    62.3  6345.1    60.8  6377.2    61.2  7225.1    62.9  8158.3    63.3
#Mann= 6 , 1 , 0
  1873.6      .2       0  3389.3      .1       0  4731.6     .06       0
  4946.5    .035       0  5040.7     .06       0  6377.2      .2       0
Bank Sta=4946.5,5040.7
XS Rating Curve= 0 ,0
Exp/Cntr=0.3,0.1

Type RM Length L Ch R = 1 ,104687.2,542.98,538.32,533.64
BEGIN DESCRIPTION:
Cross Section 106784.0-Interpolated
END DESCRIPTION:
XS GIS Cut Line= 6
 3084206.560108713795033.8866269 3084443.880108713792337.3266269
 3084538.810108713791586.8066269 3084580.340108713790649.3866269
 3084574.410108713789818.7666269 3083969.240108713788738.9566269
#Sta/Elev= 30
  1871.8   64.83  2326.8   61.94  2736.8    61.9  2751.8   60.97  3311.8    60.6
  3397.2   62.06  3466.8   58.84  3516.8   61.45  3936.2   60.49  4561.2   61.56
  4583.9   60.52  4620.2   58.42  4650.2   59.52  4710.2   58.45  4845.2   61.07
  4865.2   62.37  4905.2   62.31  4925.2   59.83  4931.4   60.51 4993.84   46.43
 5008.12   46.11  5011.2   48.52  5054.6    54.7  5066.5   59.16  5075.2   63.02
  5290.2   60.45  5524.8   59.87  6439.8   59.27    7080   61.25  8343.5   62.26
#Mann= 7 , 1 , 0
  1871.8     .15       0  3397.2     .08       0  4583.9     .06       0
  4931.4    .035       0  5066.5     .06       0  5524.8     .99       0
  6439.8      .2       0
#XS Ineff= 2 , 0
       0    4553    61.6               0
Permanent Ineff=
       F       F
Bank Sta=4931.4,5066.5
XS Rating Curve= 0 ,0
Exp/Cntr=0.3,0.1

Type RM Length L Ch R = 1 ,104148.9,381.37,298.28,187.27
BEGIN DESCRIPTION:
Cross Section  106247.1
END DESCRIPTION:
XS GIS Cut Line= 6
      3085141.33     13794340.65      3084991.32     13793360.55
      3085001.32     13792590.48      3085041.32      13791770.4
      3085021.32     13790080.24      3084351.26     13788785.12
#Sta/Elev= 30
  2585.7    63.2  3060.7    61.7  3315.7    58.9  3413.8   60.72  3470.7    58.6
  3515.7    61.1  3622.2      62  3692.2    60.8  3727.2      58  3787.2    60.8
  4187.2      60  4222.2    57.9  4347.3    61.1  4387.3    59.8  4510.2   60.07
  4842.3    60.8  4897.3    62.1    4951    60.5  4995.6   46.42  5005.8    46.1
    5008   48.51    5039   54.69  5047.5   59.15  5167.3      61  5250.7    59.6
  6720.7   59.69  6856.9    59.7  7073.7    60.1  7108.7    61.4  8316.9    62.4
#Mann= 8 , 1 , 0
  2585.7      .2       0  3413.8      .1       0  4510.2     .06       0
    4951    .035       0  5047.5     .06       0  5250.7     .99       0
  6720.7     .06       0  6856.9     .06       0
#XS Ineff= 2 , 0
       0    4344    61.1               0
Permanent Ineff=
       F       F
Bank Sta=4951,5047.5
XS Rating Curve= 0 ,0
Exp/Cntr=0.5,0.3

Type RM Length L Ch R = 1 ,103850.6,21.11,21.04,18.26
BEGIN DESCRIPTION:
Upstream Section of Bridge/Culvert/Weir
END DESCRIPTION:
XS GIS Cut Line= 6
      3085151.01     13794179.92       3085030.4     13792659.38
      3085411.19     13792020.69      3085200.55     13791895.76
      3085055.33     13790084.87      3084430.48     13788858.33
#Sta/Elev= 30
  2585.7    63.2  3060.7    61.7  3315.7    58.9  3355.7    60.6  3413.8   60.72
  3470.7    58.6  3515.7    61.1  3622.2      62  3692.2    60.8  3727.2      58
  3787.2    60.8  4187.2      60  4222.2    57.9  4347.3    61.1  4402.3    58.5
  4510.2   59.06  4897.3    62.1    4951    60.5    5000   46.05  5005.8    46.1
    5008   48.51    5039   54.69  5047.5   59.15  5167.3      61  5240.7    59.6
  6695.7   59.69  6856.9    59.7  7073.7    60.1  7108.7    61.4  8316.9    62.4
#Mann= 8 ,-1 , 0
  2585.7      .2       0  3413.8      .1       0  4510.2     .06       0
    4951    .035       0  5047.5     .06       0  5240.7     .99       0
  6695.7     .06       0  6856.9      .2       0
#XS Ineff= 2 , 0
       0    4852    61.8    5167       0      61
Permanent Ineff=
       F       F
Bank Sta=4951,5047.5
XS Rating Curve= 0 ,0
Exp/Cntr=0.5,0.3

Type RM Length L Ch R = 3 ,103840.1,,,
BEGIN DESCRIPTION:
12" DIA. PIPE
END DESCRIPTION:
Bridge Culvert--1,0,-1,-1, 0
Deck Dist Width WeirC Skew NumUp NumDn MinLoCord MaxHiCord MaxSubmerge Is_Ogee
10,1,2.6,0, 60, 60, , , 0.95, 0, 1,1,,
  2585.7  3030.7  3055.7  3060.7  3225.7  3265.7  3315.7  3335.7  3355.7  3410.7
  3425.7  3440.7  3455.7  3470.7  3485.7  3515.7  3577.2  3622.2  3692.2  3712.2
  3727.2  3742.2  3762.2  3772.2  3787.2  3892.2  3922.2  4012.2  4057.2  4187.2
  4207.2  4222.2  4252.2  4282.2  4312.2  4347.3  4367.3  4387.3  4402.3  4842.3
  4852.3  4887.3  4897.3    4951 4956.47    5039 5049.07 5056.36  5062.9  5167.3
  5233.4  6858.7  7073.7  7093.7  7108.7  7123.7  7838.7  7853.7  7868.7  8316.9
    63.2    61.1    61.5    61.7    60.6    59.1    58.9    59.6    60.6    60.8
    60.4    59.3    58.6    58.6    59.1    61.1    61.9      62    60.8    59.4
      58    58.1    59.3    60.2    60.8    60.4    60.9    59.9    60.4      60
      59    57.9    58.2    59.8    60.7    61.1      61    59.8    58.5   60.81
   61.81   61.81   62.11   60.51   60.27   59.98   59.95   59.55   59.84      61
    59.6    59.7    60.1      61    61.4    60.5    61.8    62.1    61.6    62.4
    63.2    61.1    61.5    61.7    60.6    59.1    58.9    59.6    60.6    60.8
    60.4    59.3    58.6    58.6    59.1    61.1    61.9      62    60.8    59.4
      58    58.1    59.3    60.2    60.8    60.4    60.9    59.9    60.4      60
      59    57.9    58.2    59.8    60.7    61.1      61    59.8    58.5    60.8
    61.8    61.8    62.1    60.5   59.27   58.98   59.22   59.54   59.83      61
    59.6    59.7    60.1      61    61.4    60.5    61.8    62.1    61.6    62.4
  2585.7  3030.7  3055.7  3060.7  3225.7  3265.7  3315.7  3335.7  3355.7  3410.7
  3425.7  3440.7  3455.7  3470.7  3485.7  3515.7  3577.2  3622.2  3692.2  3712.2
  3727.2  3742.2  3762.2  3772.2  3787.2  3892.2  3922.2  4012.2  4057.2  4187.2
  4207.2  4222.2  4252.2  4282.2  4312.2  4347.3  4367.3  4387.3  4402.3  4842.3
  4852.3  4887.3  4897.3    4951 4956.47    5039 5049.07 5056.36  5062.9  5167.3
  5233.4  6858.7  7073.7  7093.7  7108.7  7123.7  7838.7  7853.7  7868.7  8316.9
    63.2    61.1    61.5    61.7    60.6    59.1    58.9    59.6    60.6    60.8
    60.4    59.3    58.6    58.6    59.1    61.1    61.9      62    60.8    59.4
      58    58.1    59.3    60.2    60.8    60.4    60.9    59.9    60.4      60
      59    57.9    58.2    59.8    60.7    61.1      61    59.8    58.5   60.81
   61.81   61.81   62.11   60.51   60.27   59.98   59.95   59.55   59.84      61
    59.6    59.7    60.1      61    61.4    60.5    61.8    62.1    61.6    62.4
    63.2    61.1    61.5    61.7    60.6    59.1    58.9    59.6    60.6    60.8
    60.4    59.3    58.6    58.6    59.1    61.1    61.9      62    60.8    59.4
      58    58.1    59.3    60.2    60.8    60.4    60.9    59.9    60.4      60
      59    57.9    58.2    59.8    60.7    61.1      61    59.8    58.5    60.8
    61.8    61.8    62.1    60.5   59.27   58.98   59.22   59.54   59.83      61
    59.6    59.7    60.1      61    61.4    60.5    61.8    62.1    61.6    62.4
Pier Skew, UpSta & Num, DnSta & Num=  ,4963.4, 2 ,4963.4, 2 , 0 , 0 , 0 ,,
       1       1
   55.59   60.25
       1       1
   55.59   60.25
Pier Skew, UpSta & Num, DnSta & Num=  ,4989, 2 ,4989, 2 , 0 , 0 , 0 ,,
       1       1
   47.61   60.16
       1       1
   47.61   60.16
Pier Skew, UpSta & Num, DnSta & Num=  ,5015.3, 2 ,5015.3, 2 , 0 , 0 , 0 ,,
       1       1
   48.86   60.07
       1       1
   48.86   60.07
Pier Skew, UpSta & Num, DnSta & Num=  ,5041.4, 2 ,5041.4, 2 , 0 , 0 , 0 ,,
       1       1
   54.67   60.04
       1       1
   54.67   60.04
BR Coef= 1 , 1 , 0 ,1.25, 0 ,,,0.8,0,2,0,
WSPro=,,,, 1 ,,,, 0 ,,,, 0 ,,,,-1 ,-1 ,-1 , 0 , 0 , 0 , 0 , 0
BR U #Sta/Elev= 91
  2585.7    63.2  3030.7    61.1  3055.7    61.5  3060.7    61.7  3225.7    60.6
  3265.7    59.1  3315.7    58.9  3335.7    59.6  3355.7    60.6  3410.7    60.8
  3413.8   60.72  3425.7    60.4  3440.7    59.3  3455.7    58.6  3470.7    58.6
  3485.7    59.1  3515.7    61.1  3577.2    61.9  3622.2      62  3692.2    60.8
  3712.2    59.4  3727.2      58  3742.2    58.1  3762.2    59.3  3772.2    60.2
  3787.2    60.8  3892.2    60.4  3922.2    60.9  4012.2    59.9  4057.2    60.4
  4187.2      60  4207.2      59  4222.2    57.9  4252.2    58.2  4282.2    59.8
  4312.2    60.7  4347.3    61.1  4367.3      61  4387.3    59.8  4402.3    58.5
  4510.2   59.06  4831.1   60.74  4836.1   60.77  4842.3    60.8  4852.3    61.8
  4871.1    61.8  4887.3    61.8  4897.3    62.1  4911.1   61.64  4912.3    61.6
  4924.2   61.38  4926.1   61.32 4945.77   60.67 4945.88   60.67 4946.07   60.66
    4951    60.5 4956.47   58.84  4966.2   55.88  4992.4    47.7  4995.6   46.42
    5000   46.05  5005.8    46.1  5007.7   47.48    5008   48.51    5039   54.69
  5047.5   59.15 5049.07   59.22 5056.36   59.54 5056.47   59.55 5056.57   59.55
  5062.9   59.83  5071.1   59.92  5081.1   60.03  5101.1   60.26  5159.7   60.91
  5167.3      61  5168.4      61  5233.4    59.6  5240.7    59.6  5243.4    59.6
  6695.7   59.69  6856.9    59.7  6858.7    59.7  7073.7    60.1  7093.7      61
  7108.7    61.4  7123.7    60.5  7838.7    61.8  7853.7    62.1  7868.7    61.6
  8316.9    62.4
BR U #Mann= 8
  2585.7      .2  3413.8      .1  4510.2     .06    4951    .035  5047.5     .06
  5240.7     .99  6695.7     .06  6856.9      .2
BR U Banks=4951,5047.5
BR D #Sta/Elev= 91
  2585.7    63.2  3030.7    61.1  3055.7    61.5  3060.7    61.7  3225.7    60.6
  3265.7    59.1  3315.7    58.9  3335.7    59.6  3355.7    60.6  3410.7    60.8
  3413.8   60.72  3425.7    60.4  3440.7    59.3  3455.7    58.6  3470.7    58.6
  3485.7    59.1  3515.7    61.1  3577.2    61.9  3622.2      62  3692.2    60.8
  3712.2    59.4  3727.2      58  3742.2    58.1  3762.2    59.3  3772.2    60.2
  3787.2    60.8  3892.2    60.4  3922.2    60.9  4012.2    59.9  4057.2    60.4
  4187.2      60  4207.2      59  4222.2    57.9  4252.2    58.2  4282.2    59.8
  4312.2    60.7  4347.3    61.1  4367.3      61  4387.3    59.8  4402.3    58.5
  4510.2   59.06  4831.1   60.74  4836.1   60.77  4842.3    60.8  4852.3    61.8
  4871.1    61.8  4887.3    61.8  4897.3    62.1  4911.1   61.64  4912.3    61.6
  4924.2   61.38  4926.1   61.32 4945.77   60.67 4945.88   60.67 4946.07   60.66
    4951    60.5 4956.47   58.84  4966.2   55.88  4992.4    47.7  4995.6   46.42
    5000   46.05  5005.8    46.1  5007.7   47.48    5008   48.51    5039   54.69
  5047.5   59.15 5049.07   59.22 5056.36   59.54 5056.47   59.55 5056.57   59.55
  5062.9   59.83  5071.1   59.92  5081.1   60.03  5101.1   60.26  5159.7   60.91
  5167.3      61  5168.4      61  5233.4    59.6  5240.7    59.6  5243.4    59.6
  6695.7   59.69  6856.9    59.7  6858.7    59.7  7073.7    60.1  7093.7      61
  7108.7    61.4  7123.7    60.5  7838.7    61.8  7853.7    62.1  7868.7    61.6
  8316.9    62.4
BR D #Mann= 8
  2585.7      .2  3413.8      .1  4510.2     .06    4951    .035  5047.5     .06
  5240.7     .99  6695.7     .06  6856.9      .2
BR D Banks=4951,5047.5
BC Design=,, 0 ,, 0 ,,,,,,
BC HTab HWMax=63.2
BC Use User HTab Curves=0
BC User HTab FreeFlow(D)= 0

Type RM Length L Ch R = 1 ,103829.6,721.17,806.41,917.84
BEGIN DESCRIPTION:
Downstream Section of Bridge/Culvert/Weir
END DESCRIPTION:
XS GIS Cut Line= 6
      3085171.86     13794182.44      3085051.24      13792661.9
      3085432.03     13792023.21      3085221.39     13791898.28
      3085076.17     13790087.39      3084451.33     13788860.85
#Sta/Elev= 30
  2585.7   63.18  3060.7   61.68  3315.7   58.88  3355.7   60.58  3413.8    60.7
  3470.7   58.58  3515.7   61.08  3622.2   61.98  3692.2   60.78  3727.2   57.98
  3787.2   60.78  4187.2   59.98  4222.2   57.88  4347.3   61.08  4402.3   58.48
  4510.2   59.04  4897.3   62.08    4951   60.48    5000   46.03  5005.8   46.08
    5008   48.49    5039   54.67  5047.5   59.13  5167.3   60.98  5240.7   59.58
  6695.7   59.67  6856.9   59.68  7073.7   60.08  7108.7   61.38  8316.9   62.38
#Mann= 8 ,-1 , 0
  2585.7      .2       0  3413.8      .1       0  4510.2     .06       0
    4951    .035       0  5047.5     .06       0  5240.7     .99       0
  6695.7     .06       0  6856.9      .2       0
#XS Ineff= 2 , 0
       0    4852    61.8    5167       0      61
Permanent Ineff=
       F       F
Bank Sta=4951,5047.5
XS Rating Curve= 0 ,0
Exp/Cntr=0.5,0.3

Type RM Length L Ch R = 1 ,103023.2,170.46,168.29,164.96
BEGIN DESCRIPTION:
Cross Section 105123.0-Interpolated
END DESCRIPTION:
XS GIS Cut Line= 6
      3086034.03     13793835.42       3086045.9     13792945.47
      3086146.76     13792147.48      3086247.62     13790091.68
      3086223.89     13789919.63       3085992.5     13789617.04
#Sta/Elev= 30
  3176.6   61.69  3484.9   61.85  4061.6   62.14  4116.6   59.69  4191.6   59.78
  4221.6    61.8  4356.6   62.12  4371.6   61.63  4401.6   58.91  4486.7   59.17
  4671.6   59.73  4721.6   58.79  4791.6   59.59  4926.6   59.14    4946   59.13
  4960.8   57.01  4974.3   51.01  4992.5   45.34  5001.8   44.68  5007.8   44.94
  5011.2   48.76  5051.2   50.99  5051.3      59  5099.6      59  7076.6   59.11
  7107.9   60.12  7142.9   59.39  7197.9   59.71  7257.9   62.01  7483.8   62.04
#Mann= 9 , 1 , 0
  3176.6      .2       0  3484.9     .06       0  4486.7     .06       0
  4926.6     .06       0  4960.8    .035       0  5051.2     .06       0
  5099.6     .99       0  7076.6     .06       0  7483.8      .2       0
Bank Sta=4960.8,5051.2
XS Rating Curve= 0 ,0
Exp/Cntr=0.3,0.1

Type RM Length L Ch R = 1 ,102854.9,722.39,707.25,687.15
BEGIN DESCRIPTION:
Cross Section  104954.7
END DESCRIPTION:
XS GIS Cut Line= 6
      3086111.43     13794220.63      3086171.43     13792730.49
      3086321.44     13792340.46      3086321.44     13791820.41
      3086411.45     13790150.25      3086131.43     13789710.21
#Sta/Elev= 30
  2775.6    61.8  3471.6   61.53  4060.6    61.7  4160.6      60  4266.9    61.9
  4346.9    58.7  4398.4   58.43  4909.8    58.9  4960.8   56.73  4992.5   45.06
  5001.8    44.4  5007.8   44.66  5011.2   48.48    5038   52.32  5051.2   57.21
  5119.8    59.8  5720.1   59.23  5784.9      59  5819.9    56.4  5879.9    59.1
  6104.9      59  6149.9    57.4  6214.9      59  6404.9    59.1  6479.9    57.1
  6524.9    59.1  6749.9    57.3  6809.9    59.1    7026      60  7399.1    62.2
#Mann= 8 , 1 , 0
  2775.6      .2       0  3471.6     .06       0  4398.4     .12       0
  4960.8    .035       0  5051.2     .12       0  5720.1      .1       0
    7026     .06       0  7399.1      .2       0
#XS Ineff= 2 , 0
       0                    5695       0    59.3
Permanent Ineff=
       F       F
Bank Sta=4960.8,5051.2
XS Rating Curve= 0 ,0
Exp/Cntr=0.3,0.1

Type RM Length L Ch R = 1 ,102147.6,402.78,399.62,395.18
BEGIN DESCRIPTION:
Cross Section  104247.4
END DESCRIPTION:
XS GIS Cut Line= 6
      3087599.57     13793275.55      3087183.53     13792963.52
      3087071.52     13792131.44      3086607.47     13791043.33
      3086447.46     13790091.24      3086183.43      13789643.2
#Sta/Elev= 30
  3503.4    60.7  4023.4      60  4063.4      58  4351.5    61.2  4531.5    58.8
  4865.1    60.2  4958.8    56.9  4993.3   46.37  4995.4   43.83  5000.5   43.41
  5004.9   43.96  5006.9   47.01  5026.3   48.67  5049.9   55.94  5135.1    58.3
    5171    56.8  5739.6   58.56    5806    58.6    5881    56.2    5936    58.1
  6113.6    58.8  6233.6    56.4  6288.6    58.3  6428.6    58.5  6533.6    56.3
  6603.4   58.42  6838.6    57.3    7014    59.7  7226.4   60.15    7534    62.1
#Mann= 7 ,-1 , 0
  3503.4     .12       0  4958.8    .035       0  5049.9     .12       0
  5739.6      .1       0  6603.4      .2       0  7226.4     .99       0
    7534      .2       0
#XS Ineff= 2 , 0
       0                    5740       0    58.6
Permanent Ineff=
       F       F
Bank Sta=4958.8,5049.9
XS Rating Curve= 0 ,0
Exp/Cntr=0.3,0.1

Type RM Length L Ch R = 1 ,101748  ,26.35,26.38,26.41
XS GIS Cut Line= 6
 3087865.9309082  13793420.06427 3087422.353698713791908.6220703
 3087341.148925813791734.0316772 3086924.889099113791180.1196899
 3086469.662719713790065.4996948 3086184.468505913789617.4697266
#Sta/Elev= 30
 3321.13   59.59 3558.89   60.51 3662.92   57.73  3781.8    60.6 3841.24   58.64
 4331.63   59.51 4673.41   58.25 4732.86    56.3 4881.46   58.55 4925.94   58.13
 4951.91   55.49    5000   43.31 5014.81   48.52 5044.43   55.43  5133.1   58.67
 5678.56   58.12 5752.27   56.18 5841.21   58.21 6049.31   58.19 6123.63   55.85
 6346.59   58.15 6450.64   55.77 6614.15   58.45 6777.65   56.79 6956.02   59.42
 7162.79   59.83  7221.8   54.15  7251.3   58.32 7325.07   60.54 7516.85      62
#Mann= 6 ,-1 , 0
 3321.13     .12       0 4951.91    .035       0 5044.43     .12       0
 5678.56      .1       0 6614.15      .2       0 7162.79     .99       0
Bank Sta=4951.91,5044.43
XS Rating Curve= 0 ,0
Exp/Cntr=0.3,0.1

Type RM Length L Ch R = 5 ,101734.8,,,
BEGIN DESCRIPTION:
Drop Strucuture
END DESCRIPTION:
IW Pilot Flow=0
#Inline Weir SE= 15
    4925    53.5    4976    53.5    4976    49.5  4990.5    49.5  4990.5      48
    4997      48    4997   36.75    5000   36.75    5003   36.75    5003      48
  5009.5      48  5009.5    49.5    5024    49.5    5024    53.5    5059    53.5
IW Dist,WD,Coef,Skew,MaxSub,Min_El,Is_Ogee,SpillHt,DesHd
13.1,0.1,3.3,0,0.98,, 0 ,,,0,0,

Type RM Length L Ch R = 1 ,101721.6,119.17,111.41,101.82
XS GIS Cut Line= 6
 3087942.367675813793482.4713135 3087448.559326213791902.5856934
 3087365.148925813791722.9324951 3086937.403503413791124.0889282
  3086488.27087413790033.3380737 3086176.944091813789578.9337158
#Sta/Elev= 30
 3231.56   60.45 3604.37   60.01 3664.02   57.63 3753.49   60.38 3813.14    58.4
 4260.51    59.6 4633.31   57.97 4678.05   55.62 4722.78    58.6 4914.69   58.01
    4949   46.57    4961   46.33    4985   38.33    5000   36.75    5015   38.33
    5039   46.33    5051   46.57  5086.1   58.27 5452.85    58.7 5717.78   56.07
  5955.2   58.27 6089.58   56.14 6433.01   55.55 6552.46   58.74 6746.57   56.87
 7179.05    60.4  7238.6   54.46 7283.27   58.49  7357.7   60.68 7551.23   62.22
#Mann= 8 ,-1 , 0
 3231.56     .99       0 3753.49     .12       0 4633.31      .1       0
 4722.78     .12       0 4914.69    .045       0  5086.1     .12       0
 5452.85      .1       0 7179.05     .06       0
Bank Sta=4914.69,5086.1
XS Rating Curve= 0 ,0
Exp/Cntr=0.3,0.1

Type RM Length L Ch R = 1 ,101610.2,653.73,619.92,610.16
BEGIN DESCRIPTION:
Cross Section 103703.0-Interpolated
USACE Sims Bayou Rectification
Reach 8b Croquet to South Post Oak
File No. HSC 409-37
END DESCRIPTION:
XS GIS Cut Line= 6
      3088255.91      13793676.1      3087827.44     13792268.47
      3087530.47     13791796.03      3087112.02      13791215.6
       3086477.6     13789933.25      3086167.14      13789541.8
#Sta/Elev= 30
  2960.7    59.8  3497.2      60  3620.7    57.8  3670.7    59.5  3840.7    57.5
  4551.7   57.99  4612.1    56.5    4682   58.47 4914.69   57.91    4949   46.47
    4961   46.23    4985   38.23    5000    35.6    5015   38.23    5039   46.23
    5051   46.47  5086.1   58.17  5170.1    59.5  5540.5   56.11  5615.1    57.9
  5715.7    55.7  5985.7    58.2  6095.7    56.1  6130.7    57.8  6370.7    57.7
  6500.7    55.9  6570.7    58.2  6765.7    56.7  7343.3    60.5    7636    62.2
#Mann= 9 ,-1 , 0
  2960.7     .99       0  3497.2     .12       0  4551.7      .1       0
    4682     .12       0 4914.69    .045       0  5086.1     .12       0
  5540.5      .1       0  7343.3     .06       0    7636      .2       0
#XS Ineff= 2 , 0
       0                    5190       0    59.5
Permanent Ineff=
       F       F
Bank Sta=4914.69,5086.1
XS Rating Curve= 0 ,0
Exp/Cntr=0.3,0.1

Type RM Length L Ch R = 1 ,100990.3,527.81,566.38,584.34
BEGIN DESCRIPTION:
Cross Section  103084.9
USACE Sims Bayou Rectification
Reach 8b Croquet to South Post Oak
File No. HSC 409-37
END DESCRIPTION:
XS GIS Cut Line= 6
      3089086.38     13793734.23      3088971.44      13792745.3
      3088425.24     13791682.59        3087990.     13791394.57
      3086530.66     13789743.21      3086204.23     13789503.19
#Sta/Elev= 30
  2303.9    59.8  2388.9    59.3  2423.9    56.8  2588.9    59.6  2708.9    56.2
  2863.9    59.1  3023.9    55.9  3058.9    58.3  3206.1   59.59  3349.5    57.3
  3524.7   58.11  4394.5    57.2  4494.3    60.3  4619.3    55.6  4913.3   55.61
 4918.38   55.99    4949   45.78    4961   45.54    4985   37.54    5000    34.9
    5015   37.54    5039   45.54    5051   45.78 5091.67   59.33  5306.3      55
  5346.3    57.4  5806.1   55.53  7432.4   60.15  7625.1    62.2  7625.2    62.2
#Mann= 9 ,-1 , 0
  2303.9     .99       0  3206.1     .12       0  3524.7      .1       0
  4913.3     .12       0 4918.38    .035       0 5091.67      .1       0
  5806.1      .2       0  7432.4     .99       0  7625.1      .2       0
#XS Ineff= 2 , 0
       0                  5137.5       0    58.6
Permanent Ineff=
       F       F
Bank Sta=4918.38,5091.67
XS Rating Curve= 0 ,0
Exp/Cntr=0.3,0.1

Type RM Length L Ch R = 1 ,100423.9,158.86,176.52,197.76
BEGIN DESCRIPTION:
Cross Section 102517.0 - Interpolated
USACE Sims Bayou Rectification
Reach 8b Croquet to South Post Oak
File No. HSC 409-37
END DESCRIPTION:
XS GIS Cut Line= 6
      3089177.73     13793709.32      3089031.48     13792703.25
      3088446.57     13791073.14       3088206.9      13790615.1
      3087855.38     13790087.82      3086497.24     13789075.87
#Sta/Elev= 30
  2169.2    59.4  2264.2    56.9  2354.2    59.1  2489.2    58.9  2539.2    56.6
  2599.2    58.6  2824.2    58.3  2854.2    56.2  2944.2    59.2  3106.7   59.28
  3200.8    57.3  3401.2   58.46  4521.6    56.7  4901.6    58.7    4914   56.82
    4949   45.15    4961   44.91    4985   36.91    5000   34.28    5015   36.91
    5039   44.91    5051   45.15 5085.78   56.75  5277.4    54.6  5427.4    56.7
  5731.1    57.4  5866.1    56.1  5946.1    58.2  6069.8    58.7  7764.6    61.2
#Mann= 5 ,-1 , 0
  2169.2     .99       0  3106.7     .12       0  3401.2      .1       0
  4901.6    .035       0 5085.78      .1       0
Bank Sta=4901.6,5085.78
XS Rating Curve= 0 ,0
Exp/Cntr=0.5,0.3

Type RM Length L Ch R = 1 ,100247.4,53.56,53.43,53.35
BEGIN DESCRIPTION:
Upstream Section of Bridge/Culvert/Weir
USACE Sims Bayou Rectification
Reach 8b Croquet to South Post Oak
File No. HSC 409-37
END DESCRIPTION:
XS GIS Cut Line= 6
      3089280.03     13793678.13      3089124.03     13792674.72
       3088664.2     13791334.75      3088312.69      13790178.8
       3087638.2     13789600.66      3086569.47     13788855.03
#Sta/Elev= 30
  2131.5    59.6  2226.5    56.8  2296.5    58.9  2466.5    58.6  2496.5    56.9
  2561.5    58.7  2771.5    58.7  2816.5    56.5  2921.5    58.9  3087.7   59.23
  3182.4    57.1  3282.4    58.6  3489.7   58.14  4449.9    57.5  4691.6   55.37
 4914.58   56.43    4949   44.95    4961   44.71    4985   36.71    5000   34.08
 5008.11   36.58    5015   36.71    5039   44.71    5051   44.95 5085.98   56.61
  5304.3   54.79  5632.1    55.8  5692.1    57.6  7860.3    59.8    7967    61.7
#Mann= 5 ,-1 , 0
  2131.5     .99       0  3087.7     .12       0  3489.7      .1       0
 4914.58    .035       0 5085.98      .1       0
#XS Ineff= 2 , 0
       0 4914.58   55.79 5085.98       0    56.3
Permanent Ineff=
       F       F
Bank Sta=4914.58,5085.98
XS Rating Curve= 0 ,0
Exp/Cntr=0.5,0.3

Type RM Length L Ch R = 3 ,100220.7,,,
BEGIN DESCRIPTION:
CROOKED WOOD LANE croquet lane
Structure ID: C00-45
END DESCRIPTION:
Bridge Culvert--1,0,-1,-1, 0
Deck Dist Width WeirC Skew NumUp NumDn MinLoCord MaxHiCord MaxSubmerge Is_Ogee
10,34,2.6,0, 103, 103, , , 0.95, 0, 1,1,,
  2131.5  2181.5  2196.5  2226.5  2241.5  2296.5  2466.5  2496.5  2516.5  2561.5
  2771.5  2816.5  2846.5  2921.5  3087.7  3121.5  3157.4  3182.4  3212.4  3247.4
  3282.4  3489.7  3642.4  3657.4  3672.4  3692.4  3722.4  3737.4  4432.4  4447.4
  4449.9  4499.5  4644.9  4691.6  4750.7  4752.1  4809.8  4813.2  4859.7  4859.9
  4899.4  4900.5  4926.1 4926.21  4926.3 4926.69  4926.8 4926.91  4927.5  4954.2
  4960.1  4977.8  4977.9  4987.8  4989.2  4995.7  5003.6  5009.6  5010.8  5012.5
  5012.6  5016.3  5020.4  5043.9 5064.29  5064.4 5064.51 5064.59  5064.7  5064.8
  5070.4  5124.1    5125  5182.9  5183.7  5244.9  5248.2  5304.3  5304.9  5344.2
  5378.8  5432.5  5590.7  5612.1  5632.1  5662.1  5692.1  5822.5  5932.5  6207.5
  6377.5  6397.5  6740.3  6930.3  6945.3  7365.3  7465.3  7495.3  7515.3  7835.3
  7860.3  7910.3    7967
    59.6    59.1    58.5    56.8      57    58.9    58.6    56.9    56.9    58.7
    58.7    56.5    56.7    58.9   59.23    59.3    58.2    57.1    58.2    57.3
    58.6   58.14    57.8    58.8    58.8    57.7    57.6      58    56.8    57.5
    57.5   57.31   56.71   55.79   55.94   55.95   56.14   56.15   56.16   56.16
   56.89   56.79    56.1    56.1    56.1    56.1    56.1    56.1    56.1   56.11
   56.11   56.12   56.12   56.12   56.12   56.13   56.13   56.13   56.13   56.13
   56.13   56.13   56.13   56.14   56.15   56.15   56.15   56.15   56.15   56.15
   56.15   56.52   56.52   56.23   56.23   55.52   55.48    55.1    55.1   55.29
   55.71   55.94   56.62    56.7    55.8    56.1    57.6    57.9    57.7    58.7
    59.1    58.7    59.6    58.9    58.4    59.8    59.7    60.1    59.8    60.5
    59.8    60.5    61.7
                                                                                
                                                                                
                                                                                
                                                                                
           54.21   54.21   54.21   54.21   54.21   54.21   54.21   54.21   54.21
   54.21   54.22   54.22   54.22   54.22   54.23   54.23   54.23   54.23   54.23
   54.23   54.23   54.23   54.24   54.25   54.25   54.25   54.25   54.25   54.25
   54.25   54.25
                                                                                
                                                                                
                        
  2131.5  2181.5  2196.5  2226.5  2241.5  2296.5  2466.5  2496.5  2516.5  2561.5
  2771.5  2816.5  2846.5  2921.5  3087.7  3121.5  3157.4  3182.4  3212.4  3247.4
  3282.4  3489.7  3642.4  3657.4  3672.4  3692.4  3722.4  3737.4  4432.4  4447.4
  4449.9  4499.5  4644.9  4691.6  4750.7  4752.1  4809.8  4813.2  4859.7  4859.9
  4899.4  4900.5  4926.1 4926.21  4926.3 4926.69  4926.8 4926.91  4927.5  4954.2
  4960.1  4977.8  4977.9  4987.8  4989.2  4995.7  5003.6  5009.6  5010.8  5012.5
  5012.6  5016.3  5020.4  5043.9 5064.29  5064.4 5064.51 5064.59  5064.7  5064.8
  5070.4  5124.1    5125  5182.9  5183.7  5244.9  5248.2  5304.3  5304.9  5344.2
  5378.8  5432.5  5590.7  5612.1  5632.1  5662.1  5692.1  5822.5  5932.5  6207.5
  6377.5  6397.5  6740.3  6930.3  6945.3  7365.3  7465.3  7495.3  7515.3  7835.3
  7860.3  7910.3    7967
    59.6    59.1    58.5    56.8      57    58.9    58.6    56.9    56.9    58.7
    58.7    56.5    56.7    58.9   59.23    59.3    58.2    57.1    58.2    57.3
    58.6   58.14    57.8    58.8    58.8    57.7    57.6      58    56.8    57.5
    57.5   57.31   56.71   55.79   55.94   55.95   56.14   56.15   56.16   56.16
   56.89   56.79    56.1    56.1    56.1    56.1    56.1    56.1    56.1   56.11
   56.11   56.12   56.12   56.12   56.12   56.13   56.13   56.13   56.13   56.13
   56.13   56.13   56.13   56.14   56.15   56.15   56.15   56.15   56.15   56.15
   56.15   56.52   56.52   56.23   56.23   55.52   55.48    55.1    55.1   55.29
   55.71   55.94   56.62    56.7    55.8    56.1    57.6    57.9    57.7    58.7
    59.1    58.7    59.6    58.9    58.4    59.8    59.7    60.1    59.8    60.5
    59.8    60.5    61.7
                                                                                
                                                                                
                                                                                
                                                                                
           54.21   54.21   54.21   54.21   54.21   54.21   54.21   54.21   54.21
   54.21   54.22   54.22   54.22   54.22   54.23   54.23   54.23   54.23   54.23
   54.23   54.23   54.23   54.24   54.25   54.25   54.25   54.25   54.25   54.25
   54.25   54.25
                                                                                
                                                                                
                        
Pier Skew, UpSta & Num, DnSta & Num=  ,4960.1, 2 ,4960.1, 2 , 0 , 0 , 0 ,,
       1       1
    48.2   55.21
       1       1
   48.03   55.04
Pier Skew, UpSta & Num, DnSta & Num=  ,4987.8, 2 ,4987.8, 2 , 0 , 0 , 0 ,,
       1       1
   44.23   55.22
       1       1
   44.06   55.05
Pier Skew, UpSta & Num, DnSta & Num=  ,5016.3, 2 ,5016.3, 2 , 0 , 0 , 0 ,,
       1       1
   42.76   55.23
       1       1
   42.59   55.06
Pier Skew, UpSta & Num, DnSta & Num=  ,5043.9, 2 ,5043.9, 2 , 0 , 0 , 0 ,,
       1       1
   49.97   55.24
       1       1
    49.8   55.07
BR Coef= 1 , 1 , 0 ,1.25, 0 ,,,0.8,0,2,0,
WSPro=,,,, 1 ,,,, 0 ,,,, 0 ,,,,-1 ,-1 ,-1 , 0 , 0 , 0 , 0 , 0
BC Design=,, 0 ,, 0 ,,,,,,
BC HTab HWMax=61.7
BC Use User HTab Curves=0
BC User HTab FreeFlow(D)= 0

Type RM Length L Ch R = 1 ,100194  ,611.73,549.69,508.17
BEGIN DESCRIPTION:
Downstream Section of Bridge/Culvert/Weir
USACE Sims Bayou Rectification
Reach 8b Croquet to South Post Oak
File No. HSC 409-37
END DESCRIPTION:
XS GIS Cut Line= 6
      3089327.47     13793652.34      3089171.47     13792648.92
      3088711.64     13791308.95      3088360.13       13790153.
      3087685.64     13789574.86      3086616.91     13788829.23
#Sta/Elev= 30
  2131.5   59.43  2226.5   56.63  2296.5   58.73  2466.5   58.43  2496.5   56.73
  2561.5   58.53  2771.5   58.53  2816.5   56.33  2921.5   58.73  3087.7   59.06
  3182.4   56.93  3282.4   58.43  3489.7   57.97  4449.9   57.33  4691.6    55.2
 4913.85   56.61    4949   44.89    4961   44.65    4985   36.65    5000   34.02
 5008.11   36.52    5015   36.65    5039   44.65    5051   44.89 5086.59   56.76
  5304.3   54.62  5632.1   55.63  5692.1   57.43  7860.3   59.63    7967   61.53
#Mann= 5 ,-1 , 0
  2131.5     .99       0  3087.7     .12       0  3489.7      .1       0
 4913.85    .035       0 5086.59      .1       0
#XS Ineff= 2 , 0
       0 4913.85   55.79 5086.59       0    56.3
Permanent Ineff=
       F       F
Bank Sta=4913.85,5086.59
XS Rating Curve= 0 ,0
Exp/Cntr=0.5,0.3

Type RM Length L Ch R = 1 ,99644.3 ,361.25,367.24,358.78
BEGIN DESCRIPTION:
Cross Section 101740.3
USACE Sims Bayou Rectification
Reach 8b Croquet to South Post Oak
File No. HSC 409-37
END DESCRIPTION:
XS GIS Cut Line= 6
      3090165.98     13794332.17       3090008.2     13792322.44
      3090015.29     13791445.08      3089118.86     13790821.79
      3088460.15     13789920.66      3087466.18     13788954.32
#Sta/Elev= 30
  1057.2    63.7  1607.2    57.5  2742.2    58.6  2812.2    56.9  3130.1   60.01
  3218.1    57.6  3857.1   58.35 4892.21   56.54 4912.46   56.45    4949   44.27
    4961   44.03    4985   36.03    5000   33.39    5015   36.03    5039   44.03
    5051   44.27 5093.01   56.98  5420.3    58.4  5625.3    54.2  5700.3      57
  5930.3    57.9  5980.3      56  6055.3    58.2  6211.6    58.4  6256.6    56.4
  6356.6    57.4  6396.6    55.9  6636.6    59.6  7528.2   59.59  7548.1    59.6
#Mann= 6 ,-1 , 0
  1057.2     .99       0  3130.1     .12       0  3857.1      .1       0
 4892.21    .035       0 5093.01      .1       0  7528.2      .2       0
Bank Sta=4892.21,5093.01
XS Rating Curve= 0 ,0
Exp/Cntr=0.3,0.1

Type RM Length L Ch R = 1 ,99277   ,251.23,221.08,197.58
BEGIN DESCRIPTION:
Cross Section 101357.0 - Interpolated
USACE Sims Bayou Rectification
Reach 8b Croquet to South Post Oak
File No. HSC 409-37
END DESCRIPTION:
XS GIS Cut Line= 6
       3091270.5     13794323.86      3090521.76     13791486.89
      3089360.32     13790599.79      3088711.21     13790208.66
      3088503.02     13789948.28      3087446.34     13788925.68
#Sta/Elev= 30
   764.4    61.4   864.4    60.1   964.4    55.3  1419.4    57.8  1839.4    56.6
  2084.4    59.6  2998.6   58.47  3264.4    56.4  3404.4      59  3459.4    56.6
  3646.2   56.46  4355.3    58.1 4911.64   56.31    4949   43.86    4961   43.62
    4985   35.62    5000   32.98    5015   35.62    5039   43.62    5051   43.86
 5089.69   56.76  5521.3    56.4  5581.3    54.7  5959.1    58.1  6119.1    55.9
  6179.1      58  6362.5    58.4  6547.5    55.7  6755.7    59.5  7723.1      60
#Mann= 5 ,-1 , 0
   764.4     .99       0  2998.6     .12       0  3646.2      .1       0
 4911.64    .035       0 5089.69      .1       0
Bank Sta=4911.64,5089.69
XS Rating Curve= 0 ,0
Exp/Cntr=0.5,0.3

Type RM Length L Ch R = 1 ,99056   ,68.21,66.69,66.34
BEGIN DESCRIPTION:
Upstream Section of Bridge/Culvert/Weir
USACE Sims Bayou Rectification
Reach 8b Croquet to South Post Oak
File No. HSC 409-37
END DESCRIPTION:
XS GIS Cut Line= 6
      3091499.85     13793681.18      3090644.92     13791508.21
       3090167.2     13790815.52       3089947.1     13790625.74
        3088758.     13790153.07      3087498.41     13788906.09
#Sta/Elev= 30
  1222.3   61.14  1367.3   59.34  1762.3   60.64  1862.3   57.14  2177.3   61.24
  2387.3   57.64  2512.3   59.74    3239   57.84    3543   57.73  4305.4   56.04
  4435.4   58.24  4719.2   55.38 4911.37   56.15    4949   43.61    4961   43.37
    5000   32.73    5039   43.37    5051   43.61 5088.69   56.17  5364.1   53.96
  5934.6   57.84  6104.6   55.84  6214.6   58.24  6429.6   58.34  6559.6   55.64
  6649.6   58.54  6909.6   59.64  6974.6   57.44  7009.6   59.04  7744.6   59.84
#Mann= 6 ,-1 , 0
  1222.3     .99       0    3239     .12       0    3543      .1       0
 4911.37    .035       0 5088.69      .1       0  7744.6      .2       0
#XS Ineff= 2 , 0
       0 4911.37    55.8 5088.69       0   55.46
Permanent Ineff=
       F       F
Bank Sta=4911.37,5088.69
XS Rating Curve= 0 ,0
Exp/Cntr=0.5,0.3

Type RM Length L Ch R = 3 ,99022.7 ,,,
BEGIN DESCRIPTION:
HEATHER BROOK DRIVE
Structure ID: C00-43
END DESCRIPTION:
Bridge Culvert--1,0,-1,-1, 0
Deck Dist Width WeirC Skew NumUp NumDn MinLoCord MaxHiCord MaxSubmerge Is_Ogee
10,47,2.6,0, 60, 60, , , 0.95, 0, 1,1,,
  1222.3  1297.3  1342.3  1367.3  1762.3  1862.3  1892.3  2152.3  2177.3  2192.3
  2207.3  2387.3  2432.3  2462.3  2512.3  2547.3  3087.3  3117.3  3162.3  3182.3
  3535.4  3610.4  3845.4  3925.4  4245.4  4305.4  4435.4  4485.3    4665  4719.2
  4842.5  4915.3 4919.49 5081.79  5081.9  5114.5  5139.2  5243.6  5364.1  5470.7
  5550.7  5625.7  5934.6  6059.6  6104.6  6214.6  6429.6  6469.6  6524.6  6559.6
  6599.6  6649.6  6909.6  6949.6  6974.6  7009.6  7489.6  7534.6  7654.6  7744.6
    61.1    59.6    60.5    59.3    60.6    57.1      58    59.9    61.2    61.1
    59.9    57.6    58.2    57.7    59.7    59.1    57.7    59.4    58.7    57.8
    57.8    56.7      57    55.9    57.6      56    58.2    58.1   55.95    55.8
   55.89   56.35   56.34   56.04   56.04   55.46   55.94   54.43   53.93   54.81
    54.3    55.6    57.8    57.6    55.8    58.2    58.3    56.3    56.8    55.6
    55.9    58.5    59.6    57.4    57.4      59    58.3    59.7    59.1    59.8
    61.1    59.6    60.5    59.3    60.6    57.1      58    59.9    61.2    61.1
    59.9    57.6    58.2    57.7    59.7    59.1    57.7    59.4    58.7    57.8
    57.8    56.7      57    55.9    57.6      56    58.2    58.1   55.94   55.34
   55.83   54.98   54.44   54.14   50.51   55.45   55.93   54.42   53.92    54.8
    54.3    55.6    57.8    57.6    55.8    58.2    58.3    56.3    56.8    55.6
    55.9    58.5    59.6    57.4    57.4      59    58.3    59.7    59.1    59.8
  1222.3  1297.3  1342.3  1367.3  1762.3  1862.3  1892.3  2152.3  2177.3  2192.3
  2207.3  2387.3  2432.3  2462.3  2512.3  2547.3  3087.3  3117.3  3162.3  3182.3
  3535.4  3610.4  3845.4  3925.4  4245.4  4305.4  4435.4  4485.3    4665  4719.2
  4842.5  4915.3 4919.49 5081.79  5081.9  5114.5  5139.2  5243.6  5364.1  5470.7
  5550.7  5625.7  5934.6  6059.6  6104.6  6214.6  6429.6  6469.6  6524.6  6559.6
  6599.6  6649.6  6909.6  6949.6  6974.6  7009.6  7489.6  7534.6  7654.6  7744.6
    61.1    59.6    60.5    59.3    60.6    57.1      58    59.9    61.2    61.1
    59.9    57.6    58.2    57.7    59.7    59.1    57.7    59.4    58.7    57.8
    57.8    56.7      57    55.9    57.6      56    58.2    58.1   55.95    55.8
   55.89   56.35   56.34   56.04   56.04   55.46   55.94   54.43   53.93   54.81
    54.3    55.6    57.8    57.6    55.8    58.2    58.3    56.3    56.8    55.6
    55.9    58.5    59.6    57.4    57.4      59    58.3    59.7    59.1    59.8
   60.69   59.19   60.09   58.89   60.19   56.69   57.59   59.49   60.79   60.69
   59.49   57.19   57.79   57.29   59.29   58.69   57.29   58.99   58.29   57.39
   57.39   56.29   56.59   55.49   57.19   55.59   57.79   57.69   55.53   54.93
   55.42   54.57   54.03   53.73    50.1   55.04   55.52   54.01   53.51   54.39
   53.89   55.19   57.39   57.19   55.39   57.79   57.89   55.89   56.39   55.19
   55.49   58.09   59.19   56.99   56.99   58.59   57.89   59.29   58.69   59.39
Pier Skew, UpSta & Num, DnSta & Num=  ,4949.1, 2 ,4949.1, 2 , 0 , 0 , 0 ,,
     1.4     1.4
   46.16   55.39
     1.4     1.4
   45.75   54.98
Pier Skew, UpSta & Num, DnSta & Num=  ,4982.1, 2 ,4982.1, 2 , 0 , 0 , 0 ,,
     1.4     1.4
   40.37   55.33
     1.4     1.4
   39.96   54.92
Pier Skew, UpSta & Num, DnSta & Num=  ,5016.7, 2 ,5016.7, 2 , 0 , 0 , 0 ,,
     1.4     1.4
   42.77   55.26
     1.4     1.4
   42.36   54.85
Pier Skew, UpSta & Num, DnSta & Num=  ,5049.9, 2 ,5049.9, 2 , 0 , 0 , 0 ,,
     1.4     1.4
   46.63    55.2
     1.4     1.4
   46.22   54.79
BR Coef= 1 , 1 , 0 ,1.25, 0 ,,,0.8,0,2,0,
WSPro=,,,, 1 ,,,, 0 ,,,, 0 ,,,,-1 ,-1 ,-1 , 0 , 0 , 0 , 0 , 0
BC Design=,, 0 ,, 0 ,,,,,,
BC HTab HWMax=61.24
BC Use User HTab Curves=0
BC User HTab FreeFlow(D)= 0

Type RM Length L Ch R = 1 ,98989.3 ,767.81,875.98,972.41
BEGIN DESCRIPTION:
Downstream Section of Bridge/Culvert/Weir
USACE Sims Bayou Rectification
Reach 8b Croquet to South Post Oak
File No. HSC 409-37
END DESCRIPTION:
XS GIS Cut Line= 6
      3091547.97     13793634.56      3090693.04     13791461.59
      3090215.32      13790768.9      3089995.22     13790579.12
      3088806.12     13790106.45      3087546.53     13788859.46
#Sta/Elev= 30
  1222.3   60.66  1367.3   58.86  1762.3   60.16  1862.3   56.66  2177.3   60.76
  2387.3   57.16  2512.3   59.26    3239   57.36    3543   57.25  4305.4   55.56
  4435.4   57.76  4899.7   54.72 4910.78   56.27    4949   43.53    4961   43.29
    5000   32.66    5039   43.29    5051   43.53 5086.21   55.27  5364.1   53.48
  5934.6   57.36  6104.6   55.36  6214.6   57.76  6429.6   57.86  6559.6   55.16
  6649.6   58.06  6909.6   59.16  6974.6   56.96  7009.6   58.56  7744.6   59.36
#Mann= 6 ,-1 , 0
  1222.3     .99       0    3239     .12       0    3543      .1       0
 4910.78    .035       0 5086.21      .1       0  7744.6      .2       0
#XS Ineff= 2 , 0
       0 4910.78      55 5086.21       0   55.46
Permanent Ineff=
       F       F
Bank Sta=4910.78,5086.21
XS Rating Curve= 0 ,0
Exp/Cntr=0.5,0.3

Type RM Length L Ch R = 1 ,98113.3 ,822.91,801.4,781.44
BEGIN DESCRIPTION:
Cross Section 100195.2
USACE Sims Bayou Rectification
Reach 8b Croquet to South Post Oak
File No. HSC 409-37
END DESCRIPTION:
XS GIS Cut Line= 6
       3090839.5     13791687.51      3090830.56     13791594.79
      3090518.64     13790471.92        3090483.     13790035.24
      3089663.12     13788965.83      3088362.01     13788119.22
#Sta/Elev= 30
  3520.4    59.1  3680.2   57.82  3718.5    55.9  4138.5    54.7  4278.5    56.2
  4308.5    54.5  4373.5    56.1  4910.9   55.26    4949   42.56    4961   42.32
    4985   34.32    5000   31.68    5015   34.32    5039   42.32    5051   42.56
 5087.28   54.66    5252    54.6    5347    52.3    5422    53.9    5492    52.6
    5637    55.3    5742    53.5  5900.4   54.48    6227    56.5    6382    54.2
    6427    57.2    6522    58.1  8024.6    58.2  8079.6    61.4  8116.9    61.4
#Mann= 6 ,-1 , 0
  3520.4     .12       0  3680.2      .1       0  4910.9    .035       0
 5087.28      .2       0  5900.4      .1       0  8116.9      .2       0
Bank Sta=4910.9,5087.28
XS Rating Curve= 0 ,0
Exp/Cntr=0.3,0.1
