HEC-RAS study C100-00-00.prj: C100-00-00

--- C100-00-00.g01 (geometry) --- (continued)

Type RM Length L Ch R = 3 ,20251.6 ,,,
BEGIN DESCRIPTION:
INTERSTATE 45
Structure ID: C00-13
END DESCRIPTION:
Bridge Culvert--1,0,-1,-1, 0
Deck Dist Width WeirC Skew NumUp NumDn MinLoCord MaxHiCord MaxSubmerge Is_Ogee
10,277,2.6,0, 43, 42, , , 0.95, 0, 1,1,,
  3056.3  3255.2  3265.2  3460.2  3465.2  3735.2  3764.5  4074.5  4084.5  4286.2
  4376.2  4586.2  4588.6    4616  4662.3  4709.7  4759.2  4798.6 4801.49  4801.6
    4818  4873.1  5134.2  5170.7    5194 5194.11  5196.9  5260.9  5364.7  5440.1
  5447.8  5507.8  5517.8  5596.6  5604.1  5616.6  6285.9  6450.9  6499.1  6503.5
  6535.9  6565.9  6585.9
    37.9   36.26   36.18   34.57   34.52    32.3   32.05    29.5   29.41   27.75
   27.11   26.81    26.1   26.17   25.28    26.1   26.39    26.1   25.75   29.75
   29.86   29.96   30.42   30.49   30.53   26.53   26.98   26.79   27.93      28
   27.71   28.44   28.74   31.08    31.3   31.38   35.72   36.79    37.1      37
    35.8    36.8      36
    37.9    31.5    31.7    29.6    29.7    29.5    29.3    26.4    26.5    25.8
    27.1    26.8   26.09   26.16   25.27   26.09   26.38   26.09    25.5   25.48
   22.14   21.76   22.22   22.71    26.5   26.52   26.97   26.78   27.92   27.99
    27.7    28.4    28.2    28.4   28.29    28.1    31.4    31.5   33.62   33.86
    35.8    36.8      36
  3056.3  3255.2  3265.2  3460.2  3465.2  3735.2  3764.5  4074.5  4084.5  4286.2
  4376.2  4586.2  4588.6    4616  4662.3  4709.7  4759.2  4798.6 4801.49  4801.6
    4818  4873.1  5134.2  5170.7    5194 5194.11  5196.9  5260.9  5364.7  5440.1
  5447.8  5507.8  5517.8  5596.6  5604.1  5616.6  6285.9  6450.9  6499.1  6535.9
  6565.9  6585.9
   38.29   36.26   36.18   34.57   34.52    32.3   32.05    29.5   29.41   27.75
   27.49   27.19   26.48   26.55   25.66   26.48   26.77   26.48   25.89   29.75
   29.86   29.96   30.42   30.49   30.53   26.91   27.36   27.17   28.31   28.38
   28.09   28.79   28.74   31.08    31.3   31.38   35.72   36.79    37.1   36.19
   37.19   36.39
   38.29   31.89   32.09   29.99   30.09   29.89   29.69   26.79   26.89   26.19
   27.49   27.19   26.48   26.55   25.66   26.48   26.77   26.48   25.89   25.87
   22.53   22.15   22.61    23.1   26.89   26.91   27.36   27.17   28.31   28.38
   28.09   28.79   28.59   28.79   28.68   28.49   31.79   31.89   34.01   36.19
   37.19   36.39
Pier Skew, UpSta & Num, DnSta & Num=  ,4937.9, 2 ,4937.9, 2 , 0 , 0 , 0 ,,
       3       3
      .2   22.87
       3       3
     .59   23.26
Pier Skew, UpSta & Num, DnSta & Num=  ,5057.8, 2 ,5057.8, 2 , 0 , 0 , 0 ,,
       3       3
   -2.21   23.09
       3       3
   -1.82   23.48
Abutment Skew #Up #Dn= , 2 , 2
  4817.8  4919.1
   22.14     2.9
  4817.8  4919.1
   22.53    3.29
Abutment Skew #Up #Dn= , 2 , 2
    5071 5197.79
    3.47   26.97
    5071 5197.79
    3.86   27.36
BR Coef= 1 , 1 , 0 ,1.25, 0 ,,,0.8,-1,2,0,
WSPro=,,,, 1 ,,,, 0 ,,,, 0 ,,,,-1 ,-1 ,-1 , 0 , 0 , 0 , 0 , 0
BR U #Sta/Elev= 73
  3056.3    37.9  3255.2    31.5  3265.2    31.7  3460.2    29.6  3465.2    29.7
  3615.2    29.6  3735.2    29.5  3764.5    29.3  4074.5    26.4  4084.5    26.5
  4286.2    25.8  4376.2    27.1  4586.2    26.8  4588.6   26.09    4616   26.16
  4616.7   26.15  4661.3   25.29  4662.3   25.27  4709.7   26.09  4709.8   26.09
  4759.2   26.38  4759.6   26.38  4798.6   26.09 4801.49    25.5  4801.6   25.48
 4801.71   25.46  4817.8   22.18 4817.91   22.16    4818   22.14  4873.1   10.92
    4919    2.91  4919.1     2.9  4937.9    1.29  4941.6    1.08  4945.3   -1.21
  5007.2  -10.37    5057   -1.08  5057.8    -.67  5058.5    1.56  5070.9    3.45
    5071    3.47  5134.2   13.22  5170.7   22.71 5193.89   26.48    5194    26.5
 5194.11   26.52  5196.9   26.97 5197.59   26.97  5197.7   26.97  5197.8   26.97
  5260.9   26.78  5264.8   26.82  5314.3   27.39  5314.4   27.39  5364.7   27.92
  5365.9   27.92  5412.3   27.94  5412.7   27.94  5440.1   27.99  5447.8    27.7
  5507.8    28.4  5517.8    28.2  5596.6    28.4  5604.1   28.29  5616.6    28.1
  6285.9    31.4  6450.9    31.5  6499.1   33.62  6500.9    33.7  6503.5   33.86
  6535.9    35.8  6565.9    36.8  6585.9      36
BR U #Mann= 3
  3056.3      .1  4798.6    .035  5196.9      .1
BR U Banks=4798.6,5196.9
BR D #Sta/Elev= 73
  3056.3   38.29  3255.2   31.89  3265.2   32.09  3460.2   29.99  3465.2   30.09
  3615.2   29.99  3735.2   29.89  3764.5   29.69  4074.5   26.79  4084.5   26.89
  4286.2   26.19  4376.2   27.49  4586.2   27.19  4588.6   26.48    4616   26.55
  4616.7   26.54  4661.3   25.68  4662.3   25.66  4709.7   26.48  4709.8   26.48
  4759.2   26.77  4759.6   26.77  4798.6   26.48 4801.49   25.89  4801.6   25.87
 4801.71   25.85  4817.8   22.57 4817.91   22.55    4818   22.53  4873.1   11.31
    4919     3.3  4919.1    3.29  4937.9    1.68  4941.6    1.47  4945.3    -.82
  5007.2   -9.98    5057    -.69  5057.8    -.28  5058.5    1.95  5070.9    3.84
    5071    3.86  5134.2   13.61  5170.7    23.1 5193.89   26.87    5194   26.89
 5194.11   26.91  5196.9   27.36 5197.59   27.36  5197.7   27.36  5197.8   27.36
  5260.9   27.17  5264.8   27.21  5314.3   27.78  5314.4   27.78  5364.7   28.31
  5365.9   28.31  5412.3   28.33  5412.7   28.33  5440.1   28.38  5447.8   28.09
  5507.8   28.79  5517.8   28.59  5596.6   28.79  5604.1   28.68  5616.6   28.49
  6285.9   31.79  6450.9   31.89  6499.1   34.01  6500.9   34.09  6503.5   34.25
  6535.9   36.19  6565.9   37.19  6585.9   36.39
BR D #Mann= 3
  3056.3      .1  4798.6    .035  5196.9      .1
BR D Banks=4798.6,5196.9
BC Design=,, 0 ,, 0 ,,,,,,
BC HTab HWMax=37.95
BC Use User HTab Curves=0
BC User HTab FreeFlow(D)= 0

Type RM Length L Ch R = 1 ,20103.1 ,0.3,0.3,0.3
BEGIN DESCRIPTION:
Downstream Section of Bridge/Culvert/Weir
END DESCRIPTION:
XS GIS Cut Line= 4
      3150685.62     13815264.16      3151473.47     13814427.93
      3152420.28     13813398.19      3153099.29       13812689.
#Sta/Elev= 30
  3056.3   38.29  3255.2   31.89  3460.2   29.99  3735.2   29.89  4074.5   26.79
  4286.2   26.19  4376.2   27.49  4586.2   27.19  4588.6   26.48  4662.3   25.66
  4709.7   26.48  4798.6   26.48  4873.1   11.31    4919     3.3  4941.6    1.47
  4945.3    -.82  5007.2   -9.98    5057    -.69  5057.8    -.28  5058.5    1.95
  5134.2   13.61  5170.7    23.1  5196.9   27.36  5507.8   28.79  5616.6   28.49
  6285.9   31.79  6450.9   31.89  6535.9   36.19  6565.9   37.19  6585.9   36.39
#Mann= 3 , 1 , 0
  3056.3      .1       0  4798.6    .035       0  5196.9      .1       0
#XS Ineff= 2 , 0
       0    4808   25.69    5208       0   27.22
Permanent Ineff=
       F       F
Bank Sta=4798.6,5196.9
XS Rating Curve= 0 ,0
Exp/Cntr=0.5,0.3

Type RM Length L Ch R = 1 ,20102.8 ,23,23,23
BEGIN DESCRIPTION:
Upstream Section of Bridge/Culvert/Weir
END DESCRIPTION:
XS GIS Cut Line= 4
      3151353.35     13814489.86      3151888.66      13813989.1
      3152066.46     13813794.71      3152376.46      13813406.7
#Sta/Elev= 27
  4086.9    29.9  4236.9   27.65  4261.9   26.17  4286.9   26.42  4296.9   27.16
  4361.9   27.55  4580.9   27.39  4625.9   26.52  4640.9   25.84  4665.9   26.06
  4689.2    25.7  4724.2   25.69  4739.2   25.24 4748.72   24.58 4796.52   25.58
 4877.52   10.27 4940.22    1.65 4941.32     .59 5000.02   -9.98 5055.02     .34
 5059.72    1.42 5122.52    9.43 5198.72   25.42 5245.22   25.81    5415   28.73
    5450   30.53    5580   31.27
#Mann= 3 , 1 , 0
  4086.9      .1       0 4796.52    .035       0 5198.72      .1       0
#XS Ineff= 2 , 0
       0    4806   21.85    5197       0   22.94
Permanent Ineff=
       F       F
Bank Sta=4796.52,5198.72
XS Rating Curve= 0 ,0
Exp/Cntr=0.5,0.3

Type RM Length L Ch R = 3 ,20091.3 ,,,
BEGIN DESCRIPTION:
36" DIA. PIPE @ I-45
END DESCRIPTION:
Bridge Culvert--1,0,-1,-1, 0
Deck Dist Width WeirC Skew NumUp NumDn MinLoCord MaxHiCord MaxSubmerge Is_Ogee
10,3,2.6,0, 41, 41, , , 0.95, 0, 1,1,,
  4086.9  4236.9  4261.9  4286.9  4296.9  4361.9  4580.9  4625.9  4640.9  4665.9
  4689.2  4708.5  4724.2  4728.5  4739.2  4743.5  4744.2 4748.72  4753.5  4768.5
 4796.52 4816.12 4816.23 4816.32 4877.52 4879.92 4940.22 4941.32 5000.02 5055.02
 5059.72 5122.52 5143.42 5186.91 5187.02 5187.12 5198.72 5245.22    5415    5450
    5580
    29.9   27.65   26.17   26.42   27.16   27.55   27.39   26.52   25.84   26.06
    25.7    25.7    25.7   25.57   25.25   24.97   24.92   24.59   24.69      25
   25.59   21.89   21.86   21.85   25.85   26.07   26.17   26.17   26.26   26.35
   26.36   26.46   26.49   22.95   22.97   22.99   25.42   25.81   28.73   30.53
   31.27
    29.9   27.65   26.17   26.42   27.16   27.55   27.39   26.52   25.84   26.06
    25.7   25.69   25.69   25.56   25.24   24.96   24.91   24.58   24.68   24.99
   25.58   21.88   21.85   21.84   22.85   23.07   23.17   23.17   23.26   23.35
   23.36   23.46   23.49   22.94   22.96   22.99   25.42   25.81   28.73   30.53
   31.27
  4086.9  4236.9  4261.9  4286.9  4296.9  4361.9  4580.9  4625.9  4640.9  4665.9
  4689.2  4708.5  4724.2  4728.5  4739.2  4743.5  4744.2 4748.72  4753.5  4768.5
 4796.52 4816.12 4816.23 4816.32 4877.52 4879.92 4940.22 4941.32 5000.02 5055.02
 5059.72 5122.52 5143.42 5186.91 5187.02 5187.12 5198.72 5245.22    5415    5450
    5580
    29.9   27.65   26.17   26.42   27.16   27.55   27.39   26.52   25.84   26.06
    25.7    25.7    25.7   25.57   25.25   24.97   24.92   24.59   24.69      25
   25.59   21.89   21.86   21.85   25.85   26.07   26.17   26.17   26.26   26.35
   26.36   26.46   26.49   22.95   22.97   22.99   25.42   25.81   28.73   30.53
   31.27
    29.9   27.65   26.17   26.42   27.16   27.55   27.39   26.52   25.84   26.06
    25.7   25.69   25.69   25.56   25.24   24.96   24.91   24.58   24.68   24.99
   25.58   21.88   21.85   21.84   22.85   23.07   23.17   23.17   23.26   23.35
   23.36   23.46   23.49   22.94   22.96   22.99   25.42   25.81   28.73   30.53
   31.27
Pier Skew, UpSta & Num, DnSta & Num=  ,4822.3, 2 ,4822.3, 2 , 0 , 0 , 0 ,,
       1       1
   19.61   22.95
       1       1
   19.61   22.95
Pier Skew, UpSta & Num, DnSta & Num=  ,4859.4, 2 ,4859.4, 2 , 0 , 0 , 0 ,,
       2       2
    12.5   23.57
       2       2
    12.5   23.57
Pier Skew, UpSta & Num, DnSta & Num=  ,4916.2, 2 ,4916.2, 2 , 0 , 0 , 0 ,,
       2       2
    3.81   24.13
       2       2
    3.81   24.13
Pier Skew, UpSta & Num, DnSta & Num=  ,4986.1, 2 ,4986.1, 2 , 0 , 0 , 0 ,,
       2       2
   -8.66   24.24
       2       2
   -8.66   24.24
Pier Skew, UpSta & Num, DnSta & Num=  ,5050.6, 2 ,5050.6, 2 , 0 , 0 , 0 ,,
       2       2
   -1.67   24.34
       2       2
   -1.67   24.34
Pier Skew, UpSta & Num, DnSta & Num=  ,5110.9, 2 ,5110.9, 2 , 0 , 0 , 0 ,,
       2       2
    6.82   24.44
       2       2
    6.82   24.44
BR Coef= 1 , 1 , 0 ,1.25, 0 ,,,0.8,-1,2,0,
WSPro=,,,, 1 ,,,, 0 ,,,, 0 ,,,,-1 ,-1 ,-1 , 0 , 0 , 0 , 0 , 0
BR U #Sta/Elev= 41
  4086.9    29.9  4236.9   27.65  4261.9   26.17  4286.9   26.42  4296.9   27.16
  4361.9   27.55  4580.9   27.39  4625.9   26.52  4640.9   25.84  4665.9   26.06
  4689.2    25.7  4708.5   25.69  4724.2   25.69  4728.5   25.56  4739.2   25.24
  4743.5   24.96  4744.2   24.91 4748.72   24.58  4753.5   24.68  4768.5   24.99
 4796.52   25.58 4816.12   21.88 4816.23   21.85 4816.32   21.84 4877.52   10.27
 4879.92    9.94 4940.22    1.65 4941.32     .59 5000.02   -9.98 5055.02     .34
 5059.72    1.42 5122.52    9.43 5143.42   13.82 5186.91   22.94 5187.02   22.96
 5187.12   22.99 5198.72   25.42 5245.22   25.81    5415   28.73    5450   30.53
    5580   31.27
BR U #Mann= 3
  4086.9      .1 4796.52    .035 5198.72      .1
BR U Banks=4796.52,5198.72
BR D #Sta/Elev= 41
  4086.9    29.9  4236.9   27.65  4261.9   26.17  4286.9   26.42  4296.9   27.16
  4361.9   27.55  4580.9   27.39  4625.9   26.52  4640.9   25.84  4665.9   26.06
  4689.2    25.7  4708.5   25.69  4724.2   25.69  4728.5   25.56  4739.2   25.24
  4743.5   24.96  4744.2   24.91 4748.72   24.58  4753.5   24.68  4768.5   24.99
 4796.52   25.58 4816.12   21.88 4816.23   21.85 4816.32   21.84 4877.52   10.27
 4879.92    9.94 4940.22    1.65 4941.32     .59 5000.02   -9.98 5055.02     .34
 5059.72    1.42 5122.52    9.43 5143.42   13.82 5186.91   22.94 5187.02   22.96
 5187.12   22.99 5198.72   25.42 5245.22   25.81    5415   28.73    5450   30.53
    5580   31.27
BR D #Mann= 3
  4086.9      .1 4796.52    .035 5198.72      .1
BR D Banks=4796.52,5198.72
BC Design=,, 0 ,, 0 ,,,,,,
BC HTab HWMax=31.27
BC Use User HTab Curves=0
BC User HTab FreeFlow(D)= 0

Type RM Length L Ch R = 1 ,20079.8 ,493.4,493.4,493.4
BEGIN DESCRIPTION:
Downstream Section of Bridge/Culvert/Weir
END DESCRIPTION:
XS GIS Cut Line= 4
       3151370.3     13814505.41      3151905.62     13814004.64
      3152083.42     13813810.25      3152393.41     13813422.25
#Sta/Elev= 27
  4086.9   29.95  4236.9    27.7  4261.9   26.22  4286.9   26.47  4296.9   27.21
  4361.9    27.6  4580.9   27.44  4625.9   26.57  4640.9   25.89  4665.9   26.11
  4689.2   25.75  4724.2   25.74  4739.2   25.29 4748.72   24.63 4796.52   25.63
 4877.52   10.32 4940.22     1.7 4941.32     .64 5000.02   -9.93 5055.02     .39
 5059.72    1.47 5122.52    9.48 5198.72   25.47 5245.22   25.86    5415   28.78
    5450   30.58    5580   31.32
#Mann= 3 , 1 , 0
  4086.9      .1       0 4796.52    .035       0 5198.72      .1       0
#XS Ineff= 2 , 0
       0    4806   21.85    5197       0   22.94
Permanent Ineff=
       F       F
Bank Sta=4796.52,5198.72
XS Rating Curve= 0 ,0
Exp/Cntr=0.5,0.3

Type RM Length L Ch R = 1 ,19586.4 ,529.6,650.4,837.7
BEGIN DESCRIPTION:
Cross Section 19586.4
END DESCRIPTION:
XS GIS Cut Line= 5
       3151165.2     13815507.77      3151973.79     13814664.63
      3152457.56     13814194.68       3152547.4       13813704.
      3152554.31     13813469.03
#Sta/Elev= 30
    2908    31.2    3028    30.6    3108    28.3    3148    29.5    3473    29.5
    3523    27.2    3628    28.1    3938    26.9    3963    25.9  4076.2    27.3
  4366.2    26.4  4446.1    25.2  4711.2    24.4  4795.7    19.3  4859.3   19.35
  4867.3   18.52  4933.5   -2.21  4949.7   -5.16  4996.9   -7.48  5069.4   -1.14
  5127.9   17.39  5149.1   18.17  5150.7    16.1  5195.7    14.7  5210.7    15.4
  5254.5    20.7  5299.5    28.2    5398   30.12  5429.5    31.2  5484.6    31.2
#Mann= 7 , 1 , 0
    2908      .2       0    2908      .1       0  4446.1     .07       0
  4867.3    .035       0  5127.9     .07       0    5398      .1       0
  5484.6      .2       0
Bank Sta=4867.3,5127.9
XS Rating Curve= 0 ,0
Exp/Cntr=0.3,0.1

Type RM Length L Ch R = 1 ,18936.0 ,370.8,365.5,277.6
BEGIN DESCRIPTION:
Cross Section 18936.0 - Interpolated
END DESCRIPTION:
XS GIS Cut Line= 6
      3151209.42     13815500.55      3151809.85      13815061.7
      3152477.07     13814772.31      3152677.33     13814606.13
      3153154.55     13814231.18      3153589.15     13814128.92
#Sta/Elev= 30
  2856.6    30.8  3556.6   28.17  4327.6   26.59  4377.6      25  4481.2   24.85
  4517.6    24.8  4587.8   23.17  4627.8   21.21  4707.8   18.59  4737.8   16.81
  4797.8   18.41  4827.8   17.24  4837.8   15.17    4885   12.77  4885.5   11.34
  4905.4    6.73  4919.2    1.71  4958.7   -4.65  5031.5  -10.47  5080.1    2.15
  5083.3    4.29  5093.5    7.32  5107.8   14.72  5127.8   18.16  5147.8   23.58
  5157.8   24.93  5244.7   28.53  5544.7   29.98  5584.7    32.3  5641.2   32.43
#Mann= 6 , 1 , 0
  2856.6      .2       0  3556.6      .1       0  4481.2     .07       0
  4827.8    .035       0  5147.8     .07       0  5641.2      .2       0
Bank Sta=4827.8,5147.8
XS Rating Curve= 0 ,0
Exp/Cntr=0.5,0.3

Type RM Length L Ch R = 1 ,18570.5 ,32,32,32
BEGIN DESCRIPTION:
Upstream Section of Bridge/Culvert/Weir
END DESCRIPTION:
XS GIS Cut Line= 6
        3151333.     13815639.55      3152969.31     13814946.03
      3153141.55     13814727.39      3153183.39     13814648.39
      3153404.64     13814344.12      3153577.15     13814247.08
#Sta/Elev= 30
  2823.5   31.45  2948.5   30.35  2988.5   28.55  3138.5   29.75  3448.5   27.75
  3483.5   26.35  3728.5   24.65  3773.5   22.85  3838.5   24.75  3983.5   23.65
  4393.5   25.15  4428.5   23.55  4527.4   24.99    4563   25.24  4607.4   26.44
  4702.9   20.27  4863.1    17.6  4919.2     .03  4958.7   -6.33  5031.5  -12.15
  5080.1     .47  5083.3    2.61    5120   15.37  5120.9   13.82  5141.7   24.32
  5171.7   22.95  5235.5   25.82  5365.6   28.34  5404.4   31.05  5542.6   31.35
#Mann= 6 , 1 , 0
  2823.5      .2       0  4527.4      .1       0    4563     .07       0
  4863.1    .035       0  5141.7     .07       0  5542.6      .2       0
#XS Ineff= 2 , 0
       0    4802   19.69    5147       0   24.03
Permanent Ineff=
       F       F
Bank Sta=4863.1,5141.7
XS Rating Curve= 0 ,0
Exp/Cntr=0.5,0.3

Type RM Length L Ch R = 3 ,18554.5 ,,,
BEGIN DESCRIPTION:
GLENBROOK GOLFCOURSE FOOTBRIDGE #3 (DS TO US)
Structure ID: C00-12
END DESCRIPTION:
Bridge Culvert--1,0,-1,-1, 0
Deck Dist Width WeirC Skew NumUp NumDn MinLoCord MaxHiCord MaxSubmerge Is_Ogee
10,12,2.6,0, 43, 44, , , 0.95, 0, 1,1,,
  2823.5  2948.5  2988.5  3023.5  3138.5  3333.5  3448.5  3483.5  3728.5  3773.5
  3838.5  3938.5  3953.5  3983.5  4218.5  4248.5  4393.5  4413.5  4428.5  4453.5
  4577.6  4577.7  4607.4  4654.4  4702.9  4761.4 4812.41  4812.5 5136.26 5136.59
  5136.7  5141.7  5163.6  5171.7  5235.5  5283.7  5331.7  5336.6  5365.6  5369.4
  5389.4  5404.4  5542.6
    31.4    30.3    28.5    28.4    29.7    28.3    27.7    26.3    24.6    22.8
    24.7    24.8      24    23.6    25.1    24.9    25.1    24.4    23.5    24.4
   25.31    26.3    26.4   23.42   21.24   19.71   21.56   21.56   24.34   24.34
   24.34   24.29   24.08   24.25   25.78   26.73   28.51   28.04   28.29    28.9
    30.3      31    31.3
    31.4    30.3    28.5    28.4    29.7    28.3    27.7    26.3    24.6    22.8
    24.7    24.8      24    23.6    25.1    24.9    25.1    24.4    23.5    24.4
    25.3   26.29   26.39   23.41   20.22   18.82   18.18   20.56   23.34   23.34
   21.75   24.27   23.27    22.9   25.77   26.73   27.85   27.92   28.29    28.9
    30.3      31    31.3
  2823.5  2948.5  2958.5  2988.5  3023.5  3138.5  3333.5  3448.5  3483.5  3728.5
  3773.5  3838.5  3938.5  3953.5  3983.5  4218.5  4248.5  4393.5  4413.5  4428.5
  4453.5  4577.6  4577.7  4607.4  4654.4  4702.9  4761.4 4812.41  4812.5 5136.26
 5136.59  5136.7  5141.7  5163.6  5171.7  5235.5  5283.7  5331.7  5336.6  5365.6
  5369.4  5389.4  5404.4  5542.6
    31.6    30.5    30.1    28.7    28.6    29.9    28.5    27.9    26.5    24.8
      23    24.9      25    24.2    23.8    25.3    25.1    25.3    24.6    23.7
    24.6    25.5   26.49   26.59   23.61   21.24   19.71   21.56   21.56   24.34
   24.34   24.34   24.47   24.08   24.25   25.97   26.93   28.51   28.12   28.49
    29.1    30.5    31.2    31.5
    31.6    30.5    30.1    28.7    28.6    29.9    28.5    27.9    26.5    24.8
      23    24.9      25    24.2    23.8    25.3    25.1    25.3    24.6    23.7
    24.6    25.5   26.49   26.59   23.61   20.42   19.02   18.38   20.76   23.54
   23.54   21.95   24.47   23.47    23.1   25.97   26.93   28.05   28.12   28.49
    29.1    30.5    31.2    31.5
Pier Skew, UpSta & Num, DnSta & Num=  ,4885.5, 2 ,4885.5, 2 , 0 , 0 , 0 ,,
       2       2
    8.38   22.19
       2       2
    8.58   22.39
Pier Skew, UpSta & Num, DnSta & Num=  ,4958.7, 2 ,4958.7, 2 , 0 , 0 , 0 ,,
       2       2
   -7.47   22.82
       2       2
   -7.27   23.02
Pier Skew, UpSta & Num, DnSta & Num=  ,5031.5, 2 ,5031.5, 2 , 0 , 0 , 0 ,,
       2       2
  -13.13   23.44
       2       2
  -12.93   23.64
Pier Skew, UpSta & Num, DnSta & Num=  ,5104.2, 2 ,5104.2, 2 , 0 , 0 , 0 ,,
       2       2
    8.19   24.07
       2       2
    8.39   24.27
Pier Skew, UpSta & Num, DnSta & Num=  ,5120, 2 ,5120, 2 , 0 , 0 , 0 ,,
       1       1
   13.46    24.2
       1       1
   13.66    24.4
Abutment Skew #Up #Dn= , 2 , 2
  4812.3  4905.4
   20.56       5
  4812.3  4905.4
   20.76     5.2
Abutment Skew #Up #Dn= , 2 , 2
  5093.5 5136.79
    5.63   23.34
  5093.5 5136.79
    5.83   23.54
BR Coef= 1 , 1 , 0 ,1.25, 0 ,,,0.8,-1,2,0,
WSPro=,,,, 1 ,,,, 0 ,,,, 0 ,,,,-1 ,-1 ,-1 , 0 , 0 , 0 , 0 , 0
BR U #Sta/Elev= 79
  2823.5    31.4  2948.5    30.3  2958.5    29.9  2988.5    28.5  3023.5    28.4
  3138.5    29.7  3333.5    28.3  3448.5    27.7  3483.5    26.3  3728.5    24.6
  3773.5    22.8  3793.5    23.4  3838.5    24.7  3938.5    24.8  3953.5      24
  3983.5    23.6  4218.5    25.1  4248.5    24.9  4393.5    25.1  4413.5    24.4
  4428.5    23.5  4453.5    24.4  4527.4   24.94    4563   25.19  4572.6   25.26
  4577.6    25.3  4577.7   26.29  4605.1   26.38  4607.4   26.39  4653.4   23.47
  4654.4   23.41  4702.9   20.22  4704.5   20.18  4761.4   18.82  4762.6   18.79
  4812.3   18.18 4812.41   18.18  4812.5   18.17 4818.49    18.1  4818.6    18.1
 4818.71    18.1  4863.1   17.55    4885   11.04  4885.5    9.61  4905.3    5.02
  4905.4       5  4916.8     .86  4919.2    -.02  4958.7   -6.38  5000.8  -10.14
  5031.5   -12.2  5080.1     .42  5083.3    2.56  5093.4    5.59  5093.5    5.63
  5097.8    7.21  5104.2    9.56    5120   15.32  5120.9   13.77 5136.26   21.52
 5136.37   21.58 5136.48   21.63 5136.59   21.69  5136.7   21.75  5141.7   24.27
  5163.6   23.27  5171.7    22.9  5234.6   25.73  5235.5   25.77  5280.7   26.67
  5283.7   26.73  5329.9   27.83  5331.7   27.85  5336.6   27.92  5365.6   28.29
  5369.4    28.9  5389.4    30.3  5404.4      31  5542.6    31.3
BR U #Mann= 6
  2823.5      .2  4527.4      .1    4563     .07  4863.1    .035  5141.7     .07
  5542.6      .2
BR U Banks=4863.1,5141.7
BR D #Sta/Elev= 79
  2823.5    31.6  2948.5    30.5  2958.5    30.1  2988.5    28.7  3023.5    28.6
  3138.5    29.9  3333.5    28.5  3448.5    27.9  3483.5    26.5  3728.5    24.8
  3773.5      23  3793.5    23.6  3838.5    24.9  3938.5      25  3953.5    24.2
  3983.5    23.8  4218.5    25.3  4248.5    25.1  4393.5    25.3  4413.5    24.6
  4428.5    23.7  4453.5    24.6  4527.4   25.14    4563   25.39  4572.6   25.46
  4577.6    25.5  4577.7   26.49  4605.1   26.58  4607.4   26.59  4653.4   23.67
  4654.4   23.61  4702.9   20.42  4704.5   20.38  4761.4   19.02  4762.6   18.99
  4812.3   18.38 4812.41   18.38  4812.5   18.37 4818.49    18.3  4818.6    18.3
 4818.71    18.3  4863.1   17.75    4885   11.24  4885.5    9.81  4905.3    5.22
  4905.4     5.2  4916.8    1.06  4919.2     .18  4958.7   -6.18  5000.8   -9.94
  5031.5     -12  5080.1     .62  5083.3    2.76  5093.4    5.79  5093.5    5.83
  5097.8    7.41  5104.2    9.76    5120   15.52  5120.9   13.97 5136.26   21.72
 5136.37   21.78 5136.48   21.83 5136.59   21.89  5136.7   21.95  5141.7   24.47
  5163.6   23.47  5171.7    23.1  5234.6   25.93  5235.5   25.97  5280.7   26.87
  5283.7   26.93  5329.9   28.03  5331.7   28.05  5336.6   28.12  5365.6   28.49
  5369.4    29.1  5389.4    30.5  5404.4    31.2  5542.6    31.5
BR D #Mann= 6
  2823.5      .2  4527.4      .1    4563     .07  4863.1    .035  5141.7     .07
  5542.6      .2
BR D Banks=4863.1,5141.7
BC Design=,, 0 ,, 0 ,,,,,,
BC HTab HWMax=31.45
BC Use User HTab Curves=0
BC User HTab FreeFlow(D)= 0

Type RM Length L Ch R = 1 ,18538.5 ,462.5,462.5,462.5
BEGIN DESCRIPTION:
Downstream Section of Bridge/Culvert/Weir
END DESCRIPTION:
XS GIS Cut Line= 6
      3151352.52     13815664.91      3152988.83     13814971.39
      3153161.07     13814752.75      3153202.91     13814673.75
      3153424.16     13814369.48      3153596.67     13814272.44
#Sta/Elev= 30
  2823.5   31.65  2948.5   30.55  2988.5   28.75  3138.5   29.95  3448.5   27.95
  3483.5   26.55  3728.5   24.85  3773.5   23.05  3838.5   24.95  3983.5   23.85
  4393.5   25.35  4428.5   23.75  4527.4   25.19    4563   25.44  4607.4   26.64
  4702.9   20.47  4863.1    17.8  4919.2     .23  4958.7   -6.13  5031.5  -11.95
  5080.1     .67  5083.3    2.81    5120   15.57  5120.9   14.02  5141.7   24.52
  5171.7   23.15  5235.5   26.02  5365.6   28.54  5404.4   31.25  5542.6   31.55
#Mann= 6 , 1 , 0
  2823.5      .2       0  4527.4      .1       0    4563     .07       0
  4863.1    .035       0  5141.7     .07       0  5542.6      .2       0
#XS Ineff= 2 , 0
       0    4802   19.69    5147       0   24.03
Permanent Ineff=
       F       F
Bank Sta=4863.1,5141.7
XS Rating Curve= 0 ,0
Exp/Cntr=0.5,0.3

Type RM Length L Ch R = 1 ,18076.0 ,2562.5,162.5,169.9
BEGIN DESCRIPTION:
Cross Section 18076.0 - Interpolated
END DESCRIPTION:
XS GIS Cut Line= 6
       3151382.3     13815677.81      3152952.01     13815132.98
      3153371.85      13815219.7       3153529.5     13815027.96
      3153695.67     13814908.65      3154006.71     13814836.22
#Sta/Elev= 30
  2670.2    31.2  2840.2    28.6  3315.2    26.6  3550.2    23.6  3615.2    18.6
  3660.2    21.7  3810.2    23.5  4235.2    23.9  4381.8    26.2  4451.8    21.2
  4501.8    10.3  4576.8     2.7  4616.8     7.7  4651.8    14.4  4711.8    21.7
  4750.2   22.84  4760.5    22.9  4800.5      16  4843.4    14.5  4885.7   11.17
  4922.1    -.68  4962.4   -8.87  4995.3   -9.88  5034.8   -8.25  5077.5    -.85
  5140.6   22.84  5165.3    23.2  5185.3    28.2  5195.3    28.8  5534.2    31.1
#Mann= 5 ,-1 , 0
  2670.2     .99       0  4750.2      .1       0  4843.4    .035       0
  5140.6     .07       0  5534.2      .2       0
Bank Sta=4843.4,5140.6
XS Rating Curve= 0 ,0
Exp/Cntr=0.5,0.3

Type RM Length L Ch R = 1 ,17913.5 ,34,34,34
BEGIN DESCRIPTION:
Upstream Section of Bridge/Culvert/Weir
END DESCRIPTION:
XS GIS Cut Line= 6
      3151594.83     13817146.42      3153253.48     13815849.66
      3153428.33     13815567.31      3153418.83     13815369.61
      3153463.38     13815266.63      3154069.02     13814895.03
#Sta/Elev= 30
  2085.1   32.45  2094.6   32.38  2395.1   25.45  2490.1   18.35  2535.1    9.65
  2570.1    5.25  2745.1   10.85  2810.1   18.65  2905.1   22.85  2970.1   22.05
  3080.1   24.85  3165.1   22.95  3415.1   26.05  3495.1   25.22  3725.1   27.95
  3820.1   25.05  4180.7   27.35  4649.3   26.05  4679.3   27.95  4748.7   24.09
  4853.3   23.29  4922.1     .05  4962.4   -8.14  4995.3   -9.15  5034.8   -7.52
  5077.5    -.12  5140.6   23.57  5262.7   29.64  5507.7   30.95  5543.3   30.95
#Mann= 6 , 1 , 0
  2085.1     .15       0  2094.6     .99       0  3495.1      .1       0
  4853.3    .035       0  5140.6     .07       0  5507.7      .2       0
#XS Ineff= 2 , 0
       0    4911    4.04    5150       0   24.04
Permanent Ineff=
       F       F
Bank Sta=4853.3,5140.6
XS Rating Curve= 0 ,0
Exp/Cntr=0.5,0.3

Type RM Length L Ch R = 3 ,17896.5 ,,,
BEGIN DESCRIPTION:
GLENBROOK GOLFCOURSE FOOTBRIDGE #2 (DS TO US)
Structure ID: C00-9
END DESCRIPTION:
Bridge Culvert--1,0,-1,-1, 0
Deck Dist Width WeirC Skew NumUp NumDn MinLoCord MaxHiCord MaxSubmerge Is_Ogee
10,14,2.6,0, 60, 60, , , 0.95, 0, 1,1,,
  2085.1  2125.1  2150.1  2310.1  2325.1  2395.1  2470.1  2490.1  2535.1  2565.1
  2570.1  2585.1  2600.1  2665.1  2700.1  2745.1  2750.1  2790.1  2810.1  2905.1
  2970.1  3015.1  3055.1  3080.1  3100.1  3120.1  3165.1  3380.1  3415.1  3430.1
  3455.1  3665.1  3725.1  3755.1  3820.1  4050.1  4065.1  4180.7  4415.7  4489.3
  4529.3  4589.3  4649.3  4679.3  4699.8  4748.7  4807.3  4853.3 4855.51  4855.6
  5123.8  5140.6  5215.3  5262.7  5317.8  5374.5    5401  5406.8  5440.2  5543.3
    32.5    32.2    30.3    27.5    26.7    25.5    20.5    18.4     9.7     5.5
     5.3     5.7     5.2     7.5     9.9    10.9    11.3    17.1    18.7    22.9
    22.1    23.4    23.6    24.9    24.8    23.9      23    24.4    26.1    26.2
    25.1      26      28    27.8    25.1    26.6    26.3    27.4      26    27.7
    27.7    26.1    26.1   28.01    25.6   25.12   25.25   24.07   24.02   24.02
   23.88   23.88   28.47    29.7   30.29   30.25    30.6   30.07      31      31
    32.5    32.2    30.3    27.5    26.7    25.5    20.5    18.4     9.7     5.5
     5.3     5.7     5.2     7.5     9.9    10.9    11.3    17.1    18.7    22.9
    22.1    23.4    23.6    24.9    24.8    23.9      23    24.4    26.1    26.2
    25.1      26      28    27.8    25.1    26.6    26.3    27.4      26    27.7
    27.7    26.1    26.1      28   25.59   24.14   24.96   23.34   22.62   23.02
   22.88   23.62   28.46   29.69   30.28   30.18   30.09   30.07      31      31
  2085.1  2125.1  2150.1  2310.1  2325.1  2395.1  2470.1  2490.1  2535.1  2565.1
  2570.1  2585.1  2600.1  2665.1  2700.1  2745.1  2750.1  2790.1  2810.1  2905.1
  2970.1  3015.1  3055.1  3080.1  3100.1  3120.1  3165.1  3380.1  3415.1  3430.1
  3455.1  3665.1  3725.1  3755.1  3820.1  4050.1  4065.1  4180.7  4415.7  4489.3
  4529.3  4589.3  4649.3  4679.3  4699.8  4748.7  4807.3  4853.3 4855.51  4855.6
  5123.8  5140.6  5215.3  5262.7  5317.8  5374.5    5401  5406.8  5440.2  5543.3
    32.5    32.2    30.3    27.5    26.7    25.5    20.5    18.4     9.7     5.5
     5.3     5.7     5.2     7.5     9.9    10.9    11.3    17.1    18.7    22.9
    22.1    23.4    23.6    24.9    24.8    23.9      23    24.4    26.1    26.2
    25.1      26      28    27.8    25.1    26.6    26.3    27.4      26    27.7
    27.7    26.1    26.1   28.01    25.6   25.12   25.25   24.07   24.02   24.02
   23.88   23.88   28.47    29.7   30.29   30.25    30.6   30.07      31      31
   32.09   31.79   29.89   27.09   26.29   25.09   20.09   17.99    9.29    5.09
    4.89    5.29    4.79    7.09    9.49   10.49   10.89   16.69   18.29   22.49
   21.69   22.99   23.19   24.49   24.39   23.49   22.59   23.99   25.69   25.79
   24.69   25.59   27.59   27.39   24.69   26.19   25.89   26.99   25.59   27.29
   27.29   25.69   25.69   27.59   25.18   23.73   24.55   22.93   22.21   22.61
   22.47   23.21   28.05   29.28   29.87   29.77   29.68   29.66   30.59   30.59
Pier Skew, UpSta & Num, DnSta & Num=  ,4873.2, 2 ,4873.2, 2 , 0 , 0 , 0 ,,
       1       1
   15.69   24.01
       1       1
   15.28    23.6
Pier Skew, UpSta & Num, DnSta & Num=  ,4889.1, 2 ,4889.1, 2 , 0 , 0 , 0 ,,
       2       2
    9.42      24
       2       2
    9.01   23.59
Pier Skew, UpSta & Num, DnSta & Num=  ,4962.4, 2 ,4962.4, 2 , 0 , 0 , 0 ,,
       2       2
   -9.12   23.96
       2       2
   -9.53   23.55
Pier Skew, UpSta & Num, DnSta & Num=  ,5034.8, 2 ,5034.8, 2 , 0 , 0 , 0 ,,
       2       2
   -8.51   23.93
       2       2
   -8.92   23.52
Pier Skew, UpSta & Num, DnSta & Num=  ,5108.3, 2 ,5108.3, 2 , 0 , 0 , 0 ,,
       2       2
    9.29   23.89
       2       2
    8.88   23.48
Pier Skew, UpSta & Num, DnSta & Num=  ,5123.8, 2 ,5123.8, 2 , 0 , 0 , 0 ,,
       1       1
    15.6    23.9
       1       1
   15.19   23.49
Abutment Skew #Up #Dn= , 2 , 2
  4855.4  4906.5
   23.02     5.5
  4855.4  4906.5
   22.61    5.09
Abutment Skew #Up #Dn= , 2 , 2
  5092.3 5140.29
    5.86   23.41
  5092.3 5140.29
    5.45      23
BR Coef= 1 , 1 , 0 ,1.25, 0 ,,,0.8,-1,2,0,
WSPro=,,,, 1 ,,,, 0 ,,,, 0 ,,,,-1 ,-1 ,-1 , 0 , 0 , 0 , 0 , 0
BR U #Sta/Elev= 98
  2085.1    32.5  2094.6   32.43  2125.1    32.2  2150.1    30.3  2310.1    27.5
  2325.1    26.7  2395.1    25.5  2470.1    20.5  2490.1    18.4  2535.1     9.7
  2565.1     5.5  2570.1     5.3  2585.1     5.7  2600.1     5.2  2665.1     7.5
  2700.1     9.9  2745.1    10.9  2750.1    11.3  2790.1    17.1  2810.1    18.7
  2905.1    22.9  2970.1    22.1  3015.1    23.4  3055.1    23.6  3080.1    24.9
  3100.1    24.8  3120.1    23.9  3165.1      23  3380.1    24.4  3415.1    26.1
  3430.1    26.2  3455.1    25.1  3495.1   25.27  3665.1      26  3685.1    26.6
  3690.1    26.6  3725.1      28  3755.1    27.8  3820.1    25.1  4050.1    26.6
  4065.1    26.3  4180.7    27.4  4415.7      26  4489.3    27.7  4529.3    27.7
  4589.3    26.1  4649.3    26.1  4652.2   26.28  4679.3      28  4697.9   25.81
  4699.8   25.59  4748.7   24.14  4749.3   24.15  4805.2   24.93  4807.3   24.96
  4853.3   23.34  4855.4   22.66 4855.51   22.62  4855.6   22.59  4873.2   16.89
  4885.7   11.95  4889.1   10.72 4895.39    8.83  4895.5     8.8 4895.61    8.77
  4906.4    5.53  4906.5     5.5    4919     1.5  4922.1      .1  4962.4   -8.09
  4995.3    -9.1  5034.8   -7.47  5077.5    -.07  5080.9    1.97  5092.2    5.83
  5092.3    5.86 5101.19    8.48  5101.3    8.51 5101.41    8.55  5108.3   10.58
  5123.8    16.8 5140.09   23.41  5140.2   23.46  5140.3    23.5  5140.6   23.62
  5212.3   28.27  5215.3   28.46  5262.7   29.69  5265.1   29.72  5317.8   30.28
  5320.5   30.28  5374.5   30.18  5382.3   30.17    5401   30.09  5406.8   30.07
  5440.2      31  5507.7      31  5543.3      31
BR U #Mann= 6
  2085.1     .15  2094.6     .99  3495.1      .1  4853.3    .035  5140.6     .07
  5507.7      .2
BR U Banks=4853.3,5140.6
BR D #Sta/Elev= 98
  2085.1   32.09  2094.6   32.02  2125.1   31.79  2150.1   29.89  2310.1   27.09
  2325.1   26.29  2395.1   25.09  2470.1   20.09  2490.1   17.99  2535.1    9.29
  2565.1    5.09  2570.1    4.89  2585.1    5.29  2600.1    4.79  2665.1    7.09
  2700.1    9.49  2745.1   10.49  2750.1   10.89  2790.1   16.69  2810.1   18.29
  2905.1   22.49  2970.1   21.69  3015.1   22.99  3055.1   23.19  3080.1   24.49
  3100.1   24.39  3120.1   23.49  3165.1   22.59  3380.1   23.99  3415.1   25.69
  3430.1   25.79  3455.1   24.69  3495.1   24.86  3665.1   25.59  3685.1   26.19
  3690.1   26.19  3725.1   27.59  3755.1   27.39  3820.1   24.69  4050.1   26.19
  4065.1   25.89  4180.7   26.99  4415.7   25.59  4489.3   27.29  4529.3   27.29
  4589.3   25.69  4649.3   25.69  4652.2   25.87  4679.3   27.59  4697.9    25.4
  4699.8   25.18  4748.7   23.73  4749.3   23.74  4805.2   24.52  4807.3   24.55
  4853.3   22.93  4855.4   22.25 4855.51   22.21  4855.6   22.18  4873.2   16.48
  4885.7   11.54  4889.1   10.31 4895.39    8.42  4895.5    8.39 4895.61    8.36
  4906.4    5.12  4906.5    5.09    4919    1.09  4922.1    -.31  4962.4    -8.5
  4995.3   -9.51  5034.8   -7.88  5077.5    -.48  5080.9    1.56  5092.2    5.42
  5092.3    5.45 5101.19    8.07  5101.3     8.1 5101.41    8.14  5108.3   10.17
  5123.8   16.39 5140.09      23  5140.2   23.05  5140.3   23.09  5140.6   23.21
  5212.3   27.86  5215.3   28.05  5262.7   29.28  5265.1   29.31  5317.8   29.87
  5320.5   29.87  5374.5   29.77  5382.3   29.76    5401   29.68  5406.8   29.66
  5440.2   30.59  5507.7   30.59  5543.3   30.59
BR D #Mann= 6
  2085.1     .15  2094.6     .99  3495.1      .1  4853.3    .035  5140.6     .07
  5507.7      .2
BR D Banks=4853.3,5140.6
BC Design=,, 0 ,, 0 ,,,,,,
BC HTab HWMax=32.45
BC Use User HTab Curves=0
BC User HTab FreeFlow(D)= 0

Type RM Length L Ch R = 1 ,17879.5 ,170.7,391.3,391.3
BEGIN DESCRIPTION:
Downstream Section of Bridge/Culvert/Weir
END DESCRIPTION:
XS GIS Cut Line= 6
       3151611.9     13817175.83      3153270.54     13815879.06
      3153445.39     13815596.71      3153435.89     13815399.01
      3153480.44     13815296.03      3154086.08     13814924.43
#Sta/Elev= 30
  2085.1   32.12  2094.6   32.05  2395.1   25.12  2490.1   18.02  2535.1    9.32
  2570.1    4.92  2745.1   10.52  2810.1   18.32  2905.1   22.52  2970.1   21.72
  3080.1   24.52  3165.1   22.62  3415.1   25.72  3495.1   24.89  3725.1   27.62
  3820.1   24.72  4180.7   27.02  4649.3   25.72  4679.3   27.62  4748.7   23.76
  4853.3   22.96  4922.1    -.28  4962.4   -8.47  4995.3   -9.48  5034.8   -7.85
  5077.5    -.45  5140.6   23.24  5262.7   29.31  5507.7   30.62  5543.3   30.62
#Mann= 6 ,-1 , 0
  2085.1     .15       0  2094.6     .99       0  3495.1      .1       0
  4853.3    .035       0  5140.6     .07       0  5507.7      .2       0
#XS Ineff= 2 , 0
       0    4911    4.04    5150       0   24.04
Permanent Ineff=
       F       F
Bank Sta=4853.3,5140.6
XS Rating Curve= 0 ,0
Exp/Cntr=0.5,0.3

Type RM Length L Ch R = 1 ,17488.2 ,32,32,32
BEGIN DESCRIPTION:
Upstream Section of Bridge/Culvert/Weir
END DESCRIPTION:
XS GIS Cut Line= 6
      3151750.29     13817252.56      3153294.09      13815881.8
      3153577.67     13815670.98      3153845.54     13815532.35
      3154044.92     13815427.12      3154275.32     13815298.96
#Sta/Elev= 30
  2313.9   30.87  2401.5      30  2513.9   28.47  2813.9   16.27  2853.9   13.27
  2878.9    7.27  2973.9    3.17  3003.9    4.97  3053.9   18.27  3083.9   21.87
  3402.1   24.08  3763.9   28.07  4108.9   26.17  4444.6   28.47  4621.9   26.12
  4700.3   27.68  4798.3   27.34  4856.9   23.64    4891   10.02  4921.6     .14
  4964.3   -7.07  5036.1   -8.21  5079.5     .11  5109.1   10.19  5142.5    23.6
  5225.5   30.64  5275.3   31.68  5333.7   28.53    5476   30.87  5522.5   31.17
#Mann= 6 , 1 , 0
  2313.9     .15       0  2401.5     .99       0  3402.1      .1       0
  4856.9    .035       0  5142.5     .07       0    5476      .2       0
#XS Ineff= 2 , 0
       0    4912       4    5152       0    23.6
Permanent Ineff=
       F       F
Bank Sta=4856.9,5142.5
XS Rating Curve= 0 ,0
Exp/Cntr=0.5,0.3

Type RM Length L Ch R = 3 ,17472.2 ,,,
BEGIN DESCRIPTION:
GLENBROOK GOLFCOURSE FOOTBRIDGE #1 (DS TO US)
Structure ID: C00-8
END DESCRIPTION:
Bridge Culvert--1,0,-1,-1, 0
Deck Dist Width WeirC Skew NumUp NumDn MinLoCord MaxHiCord MaxSubmerge Is_Ogee
10,12,2.6,0, 57, 57, , , 0.95, 0, 1,1,,
  2313.9  2338.9  2453.9  2473.9  2513.9  2633.9  2713.9  2728.9  2813.9  2848.9
  2853.9  2863.9  2873.9  2878.9  2908.9  2933.9  2973.9  2993.9  2998.9  3003.9
  3008.9  3043.9  3053.9  3068.9  3083.9  3318.9  3398.9  3433.9  3548.9  3763.9
  3903.9  4108.9  4208.9  4348.9  4359.6  4379.6  4444.6    4556  4621.9  4651.4
  4700.3  4749.5  4798.3  4856.9  4858.5  5124.7 5141.59  5142.5  5171.4  5225.5
  5275.3  5330.5  5333.7  5356.7  5361.3  5430.3  5522.5
    30.9    30.3    29.8    28.6    28.5    24.1    20.5      19    16.3    13.9
    13.3    10.9     8.2     7.3     5.3     4.6     3.2     3.9     4.3       5
     6.2      16    18.3    20.7    21.9    23.9      24    25.2      25    28.1
    27.7    26.2    27.2    28.1    27.8    27.4    28.5    26.9   26.15   27.72
    27.9    28.6   27.38   24.01   23.96    23.6    23.6   23.63   26.75   30.68
   31.72   28.74    28.8    30.2   29.64    30.6    31.2
    30.9    30.3    29.8    28.6    28.5    24.1    20.5      19    16.3    13.9
    13.3    10.9     8.2     7.3     5.3     4.6     3.2     3.9     4.3       5
     6.2      16    18.3    20.7    21.9    23.9      24    25.2      25    28.1
    27.7    26.2    27.2    28.1    27.8    27.4    28.5    26.9   26.15   26.93
   27.71   26.88   27.37   23.67   23.02    22.6   23.25   23.63   26.74   30.67
   31.71   28.73   28.56   29.46   29.64    30.6    31.2
  2313.9  2338.9  2453.9  2473.9  2513.9  2633.9  2713.9  2728.9  2813.9  2848.9
  2853.9  2863.9  2873.9  2878.9  2908.9  2933.9  2973.9  2993.9  2998.9  3003.9
  3008.9  3043.9  3053.9  3068.9  3083.9  3318.9  3398.9  3433.9  3548.9  3763.9
  3903.9  4108.9  4208.9  4348.9  4359.6  4379.6  4444.6    4556  4621.9  4651.4
  4700.3  4749.5  4798.3  4856.9  4858.5  5124.7 5141.59  5141.8  5142.5  5171.4
  5225.5  5275.3  5333.7  5356.7  5361.3  5430.3  5522.5
   31.15   30.55   30.05   28.85   28.75   24.35   20.75   19.25   16.55   14.15
   13.55   11.15    8.45    7.55    5.55    4.85    3.45    4.15    4.55    5.25
    6.45   16.25   18.55   20.95   22.15   24.15   24.25   25.45   25.25   28.35
   27.95   26.45   27.45   28.35   28.05   27.65   28.75   27.15    26.4   27.72
   27.96    28.6   27.62   24.01   23.96    23.6    23.6    23.6   23.88   26.99
   30.92   31.96   28.81    30.2   29.89   30.85   31.45
   31.15   30.55   30.05   28.85   28.75   24.35   20.75   19.25   16.55   14.15
   13.55   11.15    8.45    7.55    5.55    4.85    3.45    4.15    4.55    5.25
    6.45   16.25   18.55   20.95   22.15   24.15   24.25   25.45   25.25   28.35
   27.95   26.45   27.45   28.35   28.05   27.65   28.75   27.15    26.4   27.18
   27.96   27.13   27.62   23.92   23.27   22.85    23.5   23.59   23.88   26.99
   30.92   31.96   28.81   29.71   29.89   30.85   31.45
Pier Skew, UpSta & Num, DnSta & Num=  ,4874.6, 2 ,4874.6, 2 , 0 , 0 , 0 ,,
       1       1
   15.24   23.96
       1       1
   15.49   24.21
Pier Skew, UpSta & Num, DnSta & Num=  ,4890.3, 2 ,4890.3, 2 , 0 , 0 , 0 ,,
       2       2
    8.97   23.96
       2       2
    9.22   24.21
Pier Skew, UpSta & Num, DnSta & Num=  ,4964.3, 2 ,4964.3, 2 , 0 , 0 , 0 ,,
       2       2
   -8.06   23.84
       2       2
   -7.81   24.09
Pier Skew, UpSta & Num, DnSta & Num=  ,5036.1, 2 ,5036.1, 2 , 0 , 0 , 0 ,,
       2       2
   -9.17   23.72
       2       2
   -8.92   23.97
Pier Skew, UpSta & Num, DnSta & Num=  ,5109.1, 2 ,5109.1, 2 , 0 , 0 , 0 ,,
       2       2
     8.9    23.6
       2       2
    9.15   23.85
Pier Skew, UpSta & Num, DnSta & Num=  ,5124.7, 2 ,5124.7, 2 , 0 , 0 , 0 ,,
       1       1
   14.96   23.62
       1       1
   15.21   23.87
Abutment Skew #Up #Dn= , 2 , 2
  4858.3  4908.2
   23.02    5.21
  4858.3  4908.2
   23.27    5.46
Abutment Skew #Up #Dn= , 2 , 2
  5090.5 5141.79
    4.33   23.25
  5090.5 5141.79
    4.58    23.5
BR Coef= 1 , 1 , 0 ,1.25, 0 ,,,0.8,-1,2,0,
WSPro=,,,, 1 ,,,, 0 ,,,, 0 ,,,,-1 ,-1 ,-1 , 0 , 0 , 0 , 0 , 0
BR U #Sta/Elev= 93
  2313.9    30.9  2338.9    30.3  2401.5   30.03  2453.9    29.8  2473.9    28.6
  2513.9    28.5  2633.9    24.1  2713.9    20.5  2728.9      19  2813.9    16.3
  2848.9    13.9  2853.9    13.3  2863.9    10.9  2873.9     8.2  2878.9     7.3
  2908.9     5.3  2933.9     4.6  2973.9     3.2  2993.9     3.9  2998.9     4.3
  3003.9       5  3008.9     6.2  3043.9      16  3053.9    18.3  3068.9    20.7
  3083.9    21.9  3318.9    23.9  3398.9      24  3402.1   24.11  3433.9    25.2
  3548.9      25  3763.9    28.1  3903.9    27.7  4108.9    26.2  4208.9    27.2
  4348.9    28.1  4359.6    27.8  4379.6    27.4  4444.6    28.5    4556    26.9
  4621.9   26.15  4651.4   26.93  4651.7   26.94  4700.3   27.71  4700.8    27.7
  4748.8   26.87  4749.5   26.88  4798.3   27.37  4799.8   27.28  4856.9   23.67
 4858.41   23.05  4858.5   23.02  4858.6   22.97  4874.6   16.43  4890.4   10.36
    4891   10.05 4894.59    9.04  4894.7    9.01 4894.81    8.98  4908.1    5.24
  4908.2    5.21  4918.2    1.75  4921.6     .17  4964.3   -7.04  5000.5   -7.94
  5036.1   -8.18  5079.5     .14  5081.7    1.27  5090.4     4.3  5090.5    4.33
 5104.59    8.79  5104.7    8.82 5104.81    8.86  5107.1    9.58  5109.1   10.22
  5124.7   16.15 5141.59   23.25  5141.7   23.29  5141.8   23.34  5142.5   23.63
  5171.4   26.74  5173.7   26.91  5224.6    30.6  5225.5   30.67  5275.3   31.71
  5280.4   31.43  5330.5   28.73  5333.7   28.56  5356.7   29.46  5361.3   29.64
  5430.3    30.6    5476    30.9  5522.5    31.2
BR U #Mann= 6
  2313.9     .15  2401.5     .99  3402.1      .1  4856.9    .035  5142.5     .07
    5476      .2
BR U Banks=4856.9,5142.5
BR D #Sta/Elev= 93
  2313.9   31.15  2338.9   30.55  2401.5   30.28  2453.9   30.05  2473.9   28.85
  2513.9   28.75  2633.9   24.35  2713.9   20.75  2728.9   19.25  2813.9   16.55
  2848.9   14.15  2853.9   13.55  2863.9   11.15  2873.9    8.45  2878.9    7.55
  2908.9    5.55  2933.9    4.85  2973.9    3.45  2993.9    4.15  2998.9    4.55
  3003.9    5.25  3008.9    6.45  3043.9   16.25  3053.9   18.55  3068.9   20.95
  3083.9   22.15  3318.9   24.15  3398.9   24.25  3402.1   24.36  3433.9   25.45
  3548.9   25.25  3763.9   28.35  3903.9   27.95  4108.9   26.45  4208.9   27.45
  4348.9   28.35  4359.6   28.05  4379.6   27.65  4444.6   28.75    4556   27.15
  4621.9    26.4  4651.4   27.18  4651.7   27.19  4700.3   27.96  4700.8   27.95
  4748.8   27.12  4749.5   27.13  4798.3   27.62  4799.8   27.53  4856.9   23.92
 4858.41    23.3  4858.5   23.27  4858.6   23.22  4874.6   16.68  4890.4   10.61
    4891    10.3 4894.59    9.29  4894.7    9.26 4894.81    9.23  4908.1    5.49
  4908.2    5.46  4918.2       2  4921.6     .42  4964.3   -6.79  5000.5   -7.69
  5036.1   -7.93  5079.5     .39  5081.7    1.52  5090.4    4.55  5090.5    4.58
 5104.59    9.04  5104.7    9.07 5104.81    9.11  5107.1    9.83  5109.1   10.47
  5124.7    16.4 5141.59    23.5  5141.7   23.54  5141.8   23.59  5142.5   23.88
  5171.4   26.99  5173.7   27.16  5224.6   30.85  5225.5   30.92  5275.3   31.96
  5280.4   31.68  5330.5   28.98  5333.7   28.81  5356.7   29.71  5361.3   29.89
  5430.3   30.85    5476   31.15  5522.5   31.45
BR D #Mann= 6
  2313.9     .15  2401.5     .99  3402.1      .1  4856.9    .035  5142.5     .07
    5476      .2
BR D Banks=4856.9,5142.5
BC Design=,, 0 ,, 0 ,,,,,,
BC HTab HWMax=31.68
BC Use User HTab Curves=0
BC User HTab FreeFlow(D)= 0

Type RM Length L Ch R = 1 ,17456.2 ,220.6,828.1,828.1
BEGIN DESCRIPTION:
Downstream Section of Bridge/Culvert/Weir
END DESCRIPTION:
XS GIS Cut Line= 6
      3151762.67     13817282.06      3153306.47      13815911.3
      3153590.05     13815700.48      3153857.92     13815561.85
       3154057.3     13815456.62       3154287.7     13815328.47
#Sta/Elev= 30
  2313.9   31.15  2401.5   30.28  2513.9   28.75  2813.9   16.55  2853.9   13.55
  2878.9    7.55  2973.9    3.45  3003.9    5.25  3053.9   18.55  3083.9   22.15
  3402.1   24.36  3763.9   28.35  4108.9   26.45  4444.6   28.75  4621.9    26.4
  4700.3   27.96  4798.3   27.62  4856.9   23.92    4891    10.3  4921.6     .42
  4964.3   -6.79  5036.1   -7.93  5079.5     .39  5109.1   10.47  5142.5   23.88
  5225.5   30.92  5275.3   31.96  5333.7   28.81    5476   31.15  5522.5   31.45
#Mann= 6 ,-1 , 0
  2313.9     .15       0  2401.5     .99       0  3402.1      .1       0
  4856.9    .035       0  5142.5     .07       0    5476      .2       0
#XS Ineff= 2 , 0
       0    4912       4    5152       0    23.6
Permanent Ineff=
       F       F
Bank Sta=4856.9,5142.5
XS Rating Curve= 0 ,0
Exp/Cntr=0.5,0.3

Type RM Length L Ch R = 1 ,16628.1 ,2109.3,611.8,556.7
BEGIN DESCRIPTION:
Cross Section 16628.1
END DESCRIPTION:
XS GIS Cut Line= 6
      3151838.56     13817233.97      3153743.35     13816412.79
       3153900.6     13816410.53      3154311.33     13816285.22
      3154778.54     13815962.81      3154848.89     13815652.21
#Sta/Elev= 30
  2545.7    31.7  2795.7    27.1  2830.7    24.1  3010.7    18.1  3100.7    13.6
  3160.7     3.8  3200.7     2.6  3250.7       3  3375.7    19.9  3546.4    22.7
  4215.7    22.6  4515.7    25.4  4545.7    27.7    4620    28.3    4680    26.2
    4740    27.6  4787.2    24.3  4837.2    14.3  4878.6   12.33  4927.9   -2.71
  4954.8   -6.42  5005.7   -7.79  5047.9   -6.08  5077.7   -1.42  5123.3    12.8
  5164.5    15.6  5212.4    24.7  5232.4    25.5  5989.5   28.42  6093.5    30.5
#Mann= 6 ,-1 , 0
  2545.7     .99       0  3546.4      .1       0  4878.6    .035       0
  5123.3     .07       0  5989.5      .1       0  6093.5      .2       0
Bank Sta=4878.6,5123.3
XS Rating Curve= 0 ,0
Exp/Cntr=0.3,0.1
